--- LONGRN.prj (project) ---

Proj Title=LONGRN
Current Plan=p01
Default Exp/Contr=0,0
English Units
Geom File=g01
Flow File=f01
Plan File=p01
BEGIN DESCRIPTION:
----------MODEL BY WSP USA 2022----------
AFH study
Randolph County, WV
HEC-RAS Version: RAS 6.2
Vertical Datum: NAVD88
Projection: NAD 1983 StatePlane West Virginia S FIPS 4702 (US Feet)
Terrain: 1-meter LIDAR (FEMA Region III 3DEP collected 2016-2018)
Land Use: 2019 NLCD
Hydrologic Method:
WV SIR2010-5033 regression equations
Additional Model Notes:
None
END DESCRIPTION:
DSS Export Rating Curves= 0
DSS Export Rating Curve Sorted= 0
DSS Export Volume Flow Curves= 0
DXF OffsetX= 0
DXF OffsetY= 0
DXF ScaleX= 0
DXF ScaleY= 0

--- LONGRN.p01 (plan) ---

Plan Title=Floodplain
Program Version=6.20
Short Identifier=Floodplain
Geom File=g01
Flow File=f01
Subcritical Flow
K Sum by GR= 0
Std Step Tol= 0.01
Critical Tol= 0.01
Num of Std Step Trials= 20
Max Error Tol= 0.3
Flow Tol Ratio= 0.001
Split Flow NTrial= 30
Split Flow Tol= 0.02
Split Flow Ratio= 0.02
Log Output Level= 0
Friction Slope Method= 1
Unsteady Friction Slope Method= 2
Unsteady Bridges Friction Slope Method= 1
Parabolic Critical Depth
Global Vel Dist= 0 , 0 , 0
Global Log Level= 0
CheckData=True
Encroach Param=-1 ,0,0, 0
Mapping Interval=1HOUR
Computation Time Step Use Courant=        0
Computation Time Step Use Time Series=    0
Computation Time Step Count To Double=0
Computation Time Step Max Doubling=0
Computation Time Step Max Halving=0
Computation Time Step Residence Courant=0
Run HTab= 0
Run UNet= 0
Run Sediment= 0
Run PostProcess= 0
Run WQNet= 0
Run RASMapper=-1
UNET Theta= 0
UNET Theta Warmup= 0
UNET ZTol= 0
UNET ZSATol= 0
UNET MxIter= 0
UNET Max Iter WO Improvement= 0
UNET MaxInSteps= 0
UNET DtIC= 0
UNET DtMin= 0
UNET MaxCRTS= 0
UNET WFStab= 0
UNET SFStab= 0
UNET WFX= 1
UNET SFX= 1
UNET Gravity=32.174
UNET 1D Methodology=Finite Difference
UNET DSS MLevel= 1
UNET Pardiso=0
UNET DZMax Abort= 0
UNET Use Existing IB Tables= 0
UNET Froude Reduction=False
UNET Froude Limit= 0
UNET Froude Power= 0
UNET D1 Cores= 0
UNET WindReference=Eulerian
UNET WindDragFormulation=Hsu (1988)
UNET D2 Coriolis=0
UNET D2 Cores= 0
UNET D2 Theta= 1
UNET D2 Theta Warmup= 1
UNET D2 Z Tol= 0.01
UNET D2 Volume Tol= 0.01
UNET D2 Max Iterations= 20
UNET D2 Equation= 0
UNET D2 RampUpFraction=0.1
UNET D2 TimeSlices= 1
UNET D2 Turbulence Formulation=Non-Conservative (original)
UNET D2 Eddy Viscosity=0.3
UNET D2 Transverse Eddy Viscosity=0.1
UNET D2 Smagorinsky Mixing=0
UNET D2 BCVolumeCheck=0
UNET D2 Cores=0
UNET D2 SolverType=PARDISO (Direct)
UNET D2 Minimum Iterations= 2147483647
UNET D2 Maximum Iterations= 2147483647
UNET D2 Restart Number= 10
UNET D2 Relaxation Coeff=1.3
UNET D2 SOR Precondition Iterations= 10
UNET D2 ILUT Maximum Fill= 8
UNET D2 ILUT Tolerance=1E-08
UNET D1D2 MaxIter= 0
UNET D1D2 ZTol=0.01
UNET D1D2 QTol=0.1
UNET D1D2 MinQTol=1
Write IC File= 0
Write IC File at Fixed DateTime=0
Write IC File at Sim End=0
Echo Input=False
Echo Parameters=False
Echo Output=False
Write Detailed= 0
HDF Write Warmup=0
HDF Write Time Slices=0
HDF Flush=0
HDF Compression= 1
HDF Chunk Size= 1
HDF Spatial Parts= 1
HDF Use Max Rows=0
HDF Fixed Rows= 1
Calibration Method= 0
Calibration Iterations= 20
Calibration Max Change=0.05
Calibration Tolerance=0.2
Calibration Maximum=1.5
Calibration Minimum=0.5
Calibration Optimization Method= 1
WQ AD Non Conservative
WQ ULTIMATE=-1
WQ Max Comp Step=1HOUR
WQ Output Interval=15MIN
WQ Output Selected Increments= 0
WQ Output face flow=0
WQ Output face velocity=0
WQ Output face area=0
WQ Output face dispersion=0
WQ Output cell volume=0
WQ Output cell surface area=0
WQ Output cell continuity=0
WQ Output cumulative cell continuity=0
WQ Output face conc=0
WQ Output face dconc_dx=0
WQ Output face courant=0
WQ Output face peclet=0
WQ Output face adv mass=0
WQ Output face disp mass=0
WQ Output cell mass=0
WQ Output cell source sink temp=0
WQ Output nsm pathways=0
WQ Output nsm derived pathways=0
WQ Create Restart=0
WQ Fixed Restart=0
WQ System Summary=0
WQ Write To DSS=0
Sorting and Armoring Iterations= 10
XS Update Threshold= 0.02
Bed Roughness Predictor= 0
Hydraulics Update Threshold= 0.02
Energy Slope Method= 1
Volume Change Method= 1
Sediment Retention Method= 0
Sediment TS Multiplier= 1
Warm Up Method= 0
XS Weighting Method= 0
Number of US Weighted Cross Sections= 1
Number of DS Weighted Cross Sections= 1
Upstream XS Weight=0
Main XS Weight=1
Downstream XS Weight=0
Number of DS XS's Weighted with US Boundary= 1
Upstream Boundary Weight= 1
Weight of XSs Associated with US Boundary= 0
Number of US XS's Weighted with DS Boundary= 1
Downstream Boundary Weight= 0.5
Weight of XSs Associated with DS Boundary= 0.5
Percentile Method= 0
Sediment Output Level= 3
Mass or Volume Output= 0
Output Increment Type= 1
Profile and TS Output Increment= 1
Transport Output Increment 1
XS Output Flag= 0
XS Output Increment= 10
Read HDF5 Sediment Hotstart= 0
Sediment Hotstart Type= 0
Write Gradation File= 0
Read Gradation Hotstart= 0
Write HDF5 File= 1
Write Binary Output= 1
Write DSS Sediment File= 0
DSS Sediment Output Type= 1
SV Curve= 0
Specific Gage Flag= 0
Subcell Erosion Methods= 0
Subcell Deposition Methods= 0
Advection Scheme= 1
Matrix Solver= 0
Implicit Weighting Factor= 1
Maximum Outer Loop Convergence Iterations= 5
Convergence Maximum Absolute= 0.001
Convergence RMSE= 0.0001
Grain Fractions Max Abs Error= 0.001
Max Subgrid Regions= 1
Max Subgrid Length Scale= 3.402823E+38
Initial Layer Thickness= 3.402823E+38
Min Layer Thickness= 3.402823E+38
Max Layer Thickness= 3.402823E+38
Number of Layers= 5

--- LONGRN.f01 (steady flow) ---

Flow Title=Flow
Program Version=6.20
Number of Profiles= 1
Profile Names=P100yr
River Rch & RM=LONGRN,Main,35771
     454
River Rch & RM=LONGRN,Main,33132
     514
River Rch & RM=LONGRN,Main,30056
     599
River Rch & RM=LONGRN,Main,28939
     678
River Rch & RM=LONGRN,Main,26323
     754
River Rch & RM=LONGRN,Main,22622
     839
River Rch & RM=LONGRN,Main,19593
     947
River Rch & RM=LONGRN,Main,16134
    1060
River Rch & RM=LONGRN,Main,13684
    1330
River Rch & RM=LONGRN,Main,10863
    1510
River Rch & RM=LONGRN,Main,5566
    1680
Boundary for River Rch & Prof#=LONGRN,Main            , 1
Up Type= 0
Dn Type= 3
Dn Slope=0.00736
DSS Import GetInterval= 0
DSS Import GetPeak= 0
DSS Import FillOption= 0

--- LONGRN.g01 (geometry) ---

Geom Title=Geometry
Program Version=6.20

River Reach=LONGRN          ,Main
Reach XY= 30
2230276.91194851652364.166291461     2229663.481      653420.141
     2229731.259      654637.812     2230414.574      655831.078
     2229938.429      657298.119     2230748.018      658804.735
      2231204.02      660747.025     2230834.365       662522.89
     2231434.021      663579.679     2230579.548      667823.902
     2230790.402      668213.253     2230660.056      669166.631
     2230182.111      669697.561     2229093.541      670198.082
     2228757.994      670931.872      2228168.95       671241.47
 2228475.3448689672776.509914252     2229095.582      673854.697
     2228762.374      674186.803     2229073.932      674819.504
     2228768.656      675446.2282229159.11701571678053.741116449
     2228664.574      678556.864     2228755.904       679188.35
     2229046.174      679423.082     2228651.016      679991.136
     2229242.287      680521.255     2229185.279      680921.889
     2229554.157      681379.393     2229485.971      682154.846

Type RM Length L Ch R = 1 ,35771   ,324.4,322.3,318.3
XS GIS Cut Line= 2
2230104.97807099652205.0858316712230557.37612975652638.245313194
#Sta/Elev= 30
       0 2610.67    15.5 2600.65    56.1 2584.04    67.4 2575.11    78.7 2572.12
    98.5 2558.59   115.5 2549.66   138.9 2534.84   169.2 2523.83   187.2 2518.72
   200.4 2516.33  224.71 2507.22     237 2506.19   242.8 2507.24   254.6  2508.3
   266.2 2507.45   283.5 2510.14   303.5 2509.58   389.9 2511.57   415.4 2516.36
   445.5 2525.28   460.6 2527.48   475.1 2526.76   503.1 2532.79   536.1 2542.36
   552.7 2548.25   569.3 2555.76   582.3 2558.36   596.4 2566.49   626.3 2578.09
#Mann= 5, -1 ,  0
       0     0.1       0  224.71   0.045       0   242.8     0.1       0
     500    0.06       0     540     0.1       0
Bank Sta=224.71,242.8
XS Rating Curve= 0 ,0
Exp/Cntr(USF)=0,0
Exp/Cntr=0.3,0.1

Type RM Length L Ch R = 1 ,35448   ,358.2,358.9,357.9
XS GIS Cut Line= 2
2229894.72301335652379.3888598142230410.57213574652776.085113484
#Sta/Elev= 30
       0 2610.09    36.5 2594.85    56.5 2585.47    73.6 2581.03    96.4 2577.96
   107.9 2575.03   117.9 2570.35     133 2561.09   163.3 2544.76   176.3 2542.51
   188.5 2536.29   203.7 2531.51   218.8 2523.22   228.9 2519.84     244 2516.46
   261.9 2513.92   301.8 2500.19   309.6 2498.41   321.8 2497.28   358.9 2497.52
   364.6 2496.21   380.3 2497.53   420.7 2504.77   447.3  2506.8   475.8  2513.5
   527.2 2518.21   535.7 2521.81   554.1 2525.81   602.3 2541.03   650.7 2559.79
#Mann= 5, -1 ,  0
       0     0.1       0   358.9   0.045       0   380.3     0.1       0
     480    0.06       0     640     0.1       0
Bank Sta=358.9,380.3
XS Rating Curve= 0 ,0
Exp/Cntr=0.3,0.1

Type RM Length L Ch R = 1 ,35089   ,211.8,201.1,191.9
BEGIN DESCRIPTION:
Structure XS 4
END DESCRIPTION:
XS GIS Cut Line= 3
2229710.97480515652663.5888370582229956.18460627652848.712934384
2230229.06716808652986.251467797
#Sta/Elev= 30
       0 2548.36    33.4 2539.15    61.6 2532.38   176.2 2494.22     212  2488.1
   250.5 2488.42   254.9 2487.44   261.32484.328   268.2 2481.68   274.8 2482.57
   278.32484.008   287.6 2487.17   301.4 2488.47   322.5 2486.92   337.4 2486.96
   352.7 2484.48   370.1  2485.1   392.3 2483.62   401.3 2484.39   419.2 2494.71
   423.7 2496.35   477.3 2501.03   495.4 2504.49   507.1 2508.63   522.2 2509.63
   531.2 2514.52   539.3 2517.79   596.5  2538.8   607.3 2544.96   612.8 2545.86
#Mann= 4, -1 ,  0
       0     0.1       0   261.3   0.045       0   278.3     0.1       0
  437.24    0.06       0
#XS Ineff= 2 , 0
                          330.48         2507.13
Permanent Ineff=
       F       F
Bank Sta=261.3,278.3
XS Rating Curve= 0 ,0
Exp/Cntr(USF)=0,0
Exp/Cntr=0.3,0.1

Type RM Length L Ch R = 1 ,34888   ,52.4,51.8,53.6
BEGIN DESCRIPTION:
Structure XS 3 Disconnected without IFA
END DESCRIPTION:
XS GIS Cut Line= 6
2229582.21623402652790.4540809232229724.80413741653086.258025223
2229873.06018583652992.0953998732229910.45810796652963.379138241
2229938.50654955652929.9881363442230156.50809071653060.949056054
#Sta/Elev= 30
       0  2527.3    51.9 2513.65    96.3 2496.16   105.8 2490.07   122.9 2485.23
     198 2481.23   291.7 2480.99   345.1 2477.48   430.4 2476.57   473.9 2479.41
  477.592477.529   488.1 2475.73   493.4 2477.48   498.2 2478.95   513.1 2478.54
   541.8 2479.99   578.9 2479.43   594.9 2482.08   610.7 2479.84     651 2481.64
   674.4 2480.96   685.3 2484.86   702.6 2493.89   749.1 2503.15   764.7 2510.38
   782.2 2511.54   802.5 2522.62   811.3 2526.15   839.5  2529.1   849.2 2533.12
#Mann= 9, -1 ,  0
       0     0.1       0     200    0.08       0     310    0.05       0
  378.38    0.08       0  388.38    0.05       0  477.59   0.045       0
   493.4    0.05       0  504.16     0.1       0  753.36    0.06       0
#XS Ineff= 2 , 0
          458.48 2492.81  500.36         2492.93
Permanent Ineff=
       F       F
Bank Sta=477.59,493.4
XS Rating Curve= 0 ,0
Exp/Cntr(USF)=0,0
Exp/Cntr=0.3,0.1

Type RM Length L Ch R = 1 ,34836   ,212,212.4,221.5
BEGIN DESCRIPTION:
Structure XS 2 Disconnected without IFA
END DESCRIPTION:
XS GIS Cut Line= 6
2229540.50249491652802.788585371 2229704.4606395 653144.00429225
2229774.58174349653109.9454703152229913.48831138653029.807065762
2229950.21841347652998.4195239792230132.15767258653104.671102284
#Sta/Elev= 30
       0 2518.42    13.5 2511.04      27 2507.57    82.4 2501.62    91.4 2498.32
   124.4 2491.53     147 2489.19   166.9  2485.3     260 2479.38   337.3 2478.92
   378.6 2474.54   422.4 2473.23   486.4 2474.89   533.2 2473.41   583.8 2475.93
   589.8 2475.07   597.4  2474.1  604.082475.039   610.9 2476.74   679.5 2477.75
   698.2 2482.46   713.4 2488.14   753.7 2495.46   783.1 2504.77   792.4 2509.44
     811 2511.02   829.6 2522.19   866.7 2527.83   871.4 2529.33     876 2533.25
#Mann= 8, -1 ,  0
       0     0.1       0     190    0.08       0     290    0.07       0
     310    0.05       0   569.6     0.1       0   589.8   0.045       0
  604.08     0.1       0  800.99    0.06       0
#XS Ineff= 2 , 0
          583.39 2490.52  616.27         2485.43
Permanent Ineff=
       F       F
Bank Sta=589.8,604.08
XS Rating Curve= 0 ,0
Exp/Cntr(USF)=0,0
Exp/Cntr=0.3,0.1

Type RM Length L Ch R = 1 ,34624   ,493.3,489.8,474.7
BEGIN DESCRIPTION:
Structure XS 1
END DESCRIPTION:
XS GIS Cut Line= 4
2229323.85385195653213.5721125222229521.34465391653091.527234907
2229880.82229343653253.5140724692230047.24712654653306.770019064
#Sta/Elev= 30
       0 2526.43     9.8 2522.75    28.6 2519.85    52.1 2510.51   108.5  2496.3
   152.9 2491.71   177.8 2479.16   183.6 2477.64   207.3 2475.06   232.2 2475.71
   259.7 2472.71   274.7 2475.47   393.2 2474.85   442.1 2468.27   492.6 2468.58
   502.9 2466.61   510.8 2466.79  515.942468.772   547.1 2471.45   595.5 2472.15
   608.2 2473.71   663.6 2484.97   705.6 2496.43   718.2 2502.07   726.6 2502.44
     735 2508.05   747.6 2508.46   762.5 2517.84     777 2521.55   801.2 2530.43
#Mann= 9, -1 ,  0
       0     0.1       0  292.16    0.07       0  402.16    0.05       0
  412.16    0.07       0   492.6   0.045       0  515.94    0.07       0
  622.16     0.1       0  656.45    0.07       0  726.45    0.06       0
Bank Sta=492.6,515.94
XS Rating Curve= 0 ,0
Exp/Cntr(USF)=0,0
Exp/Cntr=0.3,0.1

Type RM Length L Ch R = 1 ,34134   ,276.1,281.7,295.4
XS GIS Cut Line= 3
 2229455.1143789653674.7375818952229943.29388936653572.663684253
2230052.02478033653568.225688704
#Sta/Elev= 30
       0 2539.03     9.3 2535.02    19.1 2528.39    29.3 2523.53    50.1 2519.51
    99.2 2499.77   115.5 2494.18   119.6 2492.05   128.5 2485.15   156.4 2482.49
   181.3 2476.56   262.5 2464.27   270.8 2461.21   282.7 2454.01   303.5 2453.12
   307.6 2451.82   319.8  2450.9   336.2 2451.82   360.7 2457.85   381.1  2468.9
   397.2 2474.83   437.6 2484.69   451.7 2489.64   466.9 2491.44   483.3 2499.34
   487.4 2500.53   503.6  2500.4   511.6 2508.24   521.1 2509.63   607.6  2535.4
#Mann= 4, -1 ,  0
       0     0.1       0   307.6   0.045       0   336.2     0.1       0
  528.74    0.06       0
Bank Sta=307.6,336.2
XS Rating Curve= 0 ,0
Exp/Cntr(USF)=0,0
Exp/Cntr=0.3,0.1

Type RM Length L Ch R = 1 ,33852   ,371.8,367.7,355.2
XS GIS Cut Line= 4
2229417.05175849653821.577502823 2229610.1045649 653801.60652285
2229740.71331457 653878.601308222230049.34424667653879.025383981
#Sta/Elev= 30
       0 2564.88      36 2549.48    91.6 2530.07   111.7 2521.22   123.8  2513.2
   143.9 2510.74   188.1 2491.61   215.1 2477.34   224.3 2469.31   238.3 2459.62
   267.42445.382   270.8  2443.8   277.1  2443.5   296.62445.405   303.3 2446.43
   312.6 2450.17   331.1  2451.3   345.7 2456.02   365.2 2459.35   441.2 2457.93
   453.2 2459.59   529.2 2483.48   541.2 2489.01   561.2 2489.31   569.2 2496.56
   573.2 2498.21   601.2 2506.55   613.2 2511.51   621.2 2512.73   654.3 2522.57
#Mann= 5, -1 ,  0
       0     0.1       0   267.4   0.045       0   296.6     0.1       0
   485.7    0.06       0   575.7     0.1       0
Bank Sta=267.4,296.6
XS Rating Curve= 0 ,0
Exp/Cntr(USF)=0,0
Exp/Cntr=0.3,0.1

Type RM Length L Ch R = 1 ,33485   ,352,353.1,352.9
XS GIS Cut Line= 3
2229390.42378519654161.0841623712229585.69558938654203.245120093
2230069.43710429 654174.39814902
#Sta/Elev= 30
       0 2551.46    18.4  2546.5    46.8 2545.26    67.3 2540.93    91.8 2531.14
   139.5 2507.57   149.1 2505.67   169.6 2495.18     190 2488.33   210.3 2481.16
   226.3 2477.11   246.3 2468.62   274.4 2460.05   302.4  2441.5   321.3 2435.85
   342.5 2434.56   358.5 2435.79   378.6 2436.27   394.6 2444.83   442.7 2452.11
   511.3 2464.55   530.8 2468.95   542.9    2475   570.9 2476.22   586.9 2486.33
   590.9 2487.92     599 2488.38     615 2497.01   650.3 2512.54   684.4  2522.6
#Mann= 6, -1 ,  0
       0    0.05       0     190     0.1       0   321.3   0.045       0
   358.5     0.1       0  489.77    0.06       0  589.77     0.1       0
#XS Ineff= 2 , 0
                          362.64         2441.56
Permanent Ineff=
       F       F
Bank Sta=321.3,358.5
XS Rating Curve= 0 ,0
Exp/Cntr(USF)=0,0
Exp/Cntr=0.3,0.1

Type RM Length L Ch R = 1 ,33132   ,437.6,437,430.4
XS GIS Cut Line= 2
2229379.07800207654582.8278720152230098.03328112654502.943952121
#Sta/Elev= 30
       0 2538.91    21.2 2531.91    33.3 2529.15    45.4 2523.89    73.5 2514.56
   117.8 2498.15   137.9 2493.98   162.1 2484.92   178.2 2482.38   218.4  2470.1
   226.5 2469.01   270.8 2454.41   299.5 2442.95   327.1 2429.29   335.1 2427.49
   338.5 2425.41   343.2 2424.64   357.1 2425.43   422.7 2429.25   447.8 2436.72
   463.9 2440.36   516.3 2448.13   552.5 2455.04   572.6 2461.11   592.7 2469.26
   608.8 2469.46   612.8  2473.3   616.9 2475.72   676.2 2493.22   723.4 2508.89
#Mann= 5, -1 ,  0
       0     0.1       0   338.5   0.045       0   357.1     0.1       0
     500    0.06       0     700     0.1       0
Bank Sta=338.5,357.1
XS Rating Curve= 0 ,0
Exp/Cntr(USF)=0,0
Exp/Cntr=0.3,0.1

Type RM Length L Ch R = 1 ,32695   ,342.2,345.6,345.2
XS GIS Cut Line= 2
2229621.19955378655070.8732500482230204.79596855654724.709597176
#Sta/Elev= 30
       0 2522.96     3.5 2522.25    12.8 2516.55    26.8 2515.57   114.3 2473.06
     222 2433.33   259.2 2423.81   287.2 2418.52   304.1 2416.82   319.7  2413.3
     329 2415.13   356.9 2415.09   374.1 2413.42  383.782415.176   389.5 2418.67
   403.3 2431.49     411 2434.88   426.7 2436.15     450 2444.25   519.7 2457.48
   547.6 2466.21   563.9 2466.69   566.2 2467.22   570.8 2470.95   581.4  2474.5
   638.4 2487.99   645.3 2488.65   659.2  2493.4   673.2 2494.25   678.5 2496.24
#Mann= 6, -1 ,  0
       0    0.08       0     180     0.1       0   356.9   0.045       0
  383.78     0.1       0     470    0.06       0     640     0.1       0
Bank Sta=356.9,383.78
XS Rating Curve= 0 ,0
Exp/Cntr(USF)=0,0
Exp/Cntr=0.3,0.1

Type RM Length L Ch R = 1 ,32349   ,479.5,482.1,481.5
XS GIS Cut Line= 2
2229772.09140246655337.1529830272230351.24982169654982.113339055
#Sta/Elev= 30
       0 2509.13     9.5 2507.31    37.9 2491.73    87.3  2471.3   140.9 2452.24
   183.3 2434.01   197.2 2432.74   209.5 2427.74   225.3 2419.54  243.62  2405.5
   264.7  2405.5     288 2406.97   317.1 2404.14   328.7 2405.54   337.9 2403.39
   354.9 2409.06   366.1 2407.46   397.9 2410.73   445.8 2409.68   459.2 2411.68
   502.1 2437.67   516.2 2444.38   530.3 2448.31   553.7 2458.43   572.5 2459.64
   584.7 2468.93   628.8 2485.33   652.3 2497.44   666.3 2499.03   679.3 2504.74
#Mann= 5, -1 ,  0
       0    0.08       0     120     0.1       0  243.62   0.045       0
   264.7     0.1       0     580    0.06       0
#XS Ineff= 2 , 0
                          287.58         2465.38
Permanent Ineff=
       F       F
Bank Sta=243.62,264.7
XS Rating Curve= 0 ,0
Exp/Cntr(USF)=0,0
Exp/Cntr=0.3,0.1

Type RM Length L Ch R = 1 ,31867   ,474.9,484.4,492.7
XS GIS Cut Line= 2
2229996.21017772655692.192626998 2230553.1786192655388.189931848
#Sta/Elev= 30
       0  2503.2    72.9 2465.86   145.8    2438     164 2432.29   173.1 2427.55
   177.7 2426.27   187.9  2425.5   198.3 2419.95   206.7 2416.73   218.7 2413.36
   231.7 2407.87   256.8 2400.74  270.992390.885   273.5 2389.96   285.2 2389.56
     294 2390.91   305.3  2392.9   364.8 2396.34   378.2 2394.55   391.9 2390.06
   410.1 2392.51   432.6 2403.81   515.6 2427.59   532.3 2433.91   538.7 2437.74
   559.4 2439.22     565 2442.94   574.1 2445.18   582.9 2448.85   634.5 2462.85
#Mann= 7, -1 ,  0
       0     0.1       0     150    0.08       0  270.99   0.045       0
     294    0.08       0     350     0.1       0     540    0.06       0
     560     0.1       0
#XS Ineff= 2 , 0
                          374.76         2401.49
Permanent Ineff=
       F       F
Bank Sta=270.99,294
XS Rating Curve= 0 ,0
Exp/Cntr(USF)=0,0
Exp/Cntr=0.3,0.1

Type RM Length L Ch R = 1 ,31383   ,253.8,252.6,250.9
XS GIS Cut Line= 3
2230018.40015547655891.9024267322230428.91474381655991.757326599
2230686.31848569655958.472359977
#Sta/Elev= 30
       0 2502.76    71.8 2471.32     113 2454.89   129.4 2445.58   137.7 2444.49
   161.5 2428.03   174.7 2421.45     183 2412.44   187.1 2410.65   199.4 2408.95
   207.7 2405.58   224.1 2392.96   244.7  2383.6   261.2 2381.15   339.4 2380.11
   351.7 2378.93  357.032376.731   360.1 2375.56   372.3  2375.3   381.5 2376.76
   389.9 2380.04   409.4 2381.29   433.8 2391.38   481.3 2402.21     542 2412.43
   562.9 2418.46   583.1 2420.94   591.1 2425.19   659.7 2447.71     682 2456.42
#Mann= 5, -1 ,  0
       0    0.08       0      60     0.1       0  357.03   0.045       0
   381.5     0.1       0  662.48    0.06       0
Bank Sta=357.03,381.5
XS Rating Curve= 0 ,0
Exp/Cntr(USF)=0,0
Exp/Cntr=0.3,0.1

Type RM Length L Ch R = 1 ,31130   ,248.5,252.8,256.7
XS GIS Cut Line= 4
2229982.01547414656136.9802102752230220.78052232656214.142085598
2230407.13373064656230.1568144392230632.79581885656230.156814439
#Sta/Elev= 30
       0 2491.69    23.3 2481.13    40.1 2472.06   103.2 2443.93   115.8 2437.27
   138.5 2427.82   149.4 2420.25   153.6 2418.76     162 2418.47   166.2 2417.23
   174.6 2411.84   191.4 2403.26   208.8 2396.09   250.9  2383.1   297.5    2377
   318.6 2376.68   338.72369.272   346.7 2368.51   358.42368.944   366.7 2372.84
   370.8 2373.46   390.8 2373.06   422.9 2376.09     443 2376.89     471 2380.22
     507 2394.62     583 2414.91     595  2415.5     607 2421.01   663.6 2438.14
#Mann= 7, -1 ,  0
       0    0.08       0     100     0.1       0     200    0.08       0
  300.92     0.1       0   338.7   0.045       0   358.4     0.1       0
  597.96    0.06       0
Bank Sta=338.7,358.4
XS Rating Curve= 0 ,0
Exp/Cntr(USF)=0,0
Exp/Cntr=0.3,0.1

Type RM Length L Ch R = 1 ,30877   ,271.5,270.4,268.4
XS GIS Cut Line= 2
 2229883.0412912656269.1320484522230542.08363033656626.390690198
#Sta/Elev= 30
       0 2499.65    14.9 2489.55    28.6 2484.48    56.9 2469.61   142.8 2433.25
   159.6 2425.02     169 2418.08   183.3 2415.37   196.9 2407.55   226.7 2394.53
   251.5 2388.03   307.7 2380.97   319.8 2376.65   335.8  2373.6   347.1 2367.39
  362.442363.421   377.8 2361.87     388 2363.47   419.9 2365.72   481.8 2364.46
   501.8  2366.7   520.2 2372.77   556.4 2387.74   570.3  2389.4   579.1 2392.93
     611 2400.81   674.7 2421.73   697.2 2422.14   711.1 2432.96   749.6 2446.41
#Mann= 5, -1 ,  0
       0    0.08       0     100     0.1       0  362.44   0.045       0
     388     0.1       0     660    0.06       0
#XS Ineff= 2 , 0
                          400.52          2375.6
Permanent Ineff=
       F       F
Bank Sta=362.44,388
XS Rating Curve= 0 ,0
Exp/Cntr(USF)=0,0
Exp/Cntr=0.3,0.1

Type RM Length L Ch R = 1 ,30607   ,543,550.5,548.6
BEGIN DESCRIPTION:
Structure XS 4
END DESCRIPTION:
XS GIS Cut Line= 3
2229843.70645234656527.1572402122230290.66297544656783.392901663
2230428.97199724656813.966474904
#Sta/Elev= 30
       0 2456.88    28.2  2448.5    66.3 2432.94   101.5 2414.49   111.2 2406.58
     125 2404.17   133.7  2396.8   145.4 2389.63   157.3 2387.74   189.6 2375.67
   215.8 2369.09   235.7 2366.88   277.3    2358   295.6 2356.66   318.7 2357.97
   349.9 2355.74   355.6 2354.79     366 2355.75   378.6 2359.96   387.8 2361.26
   397.5 2360.92   480.1 2370.17   508.8 2376.37   521.3 2377.18   549.5 2386.74
     570 2396.55   595.1 2396.96   598.7 2398.45   608.5 2407.15   656.8 2425.77
#Mann= 5, -1 ,  0
       0    0.08       0      40     0.1       0   349.9   0.045       0
     366     0.1       0   595.2    0.06       0
Bank Sta=349.9,366
XS Rating Curve= 0 ,0
Exp/Cntr(USF)=0,0
Exp/Cntr=0.3,0.1

Type RM Length L Ch R = 1 ,30056   ,55,54.6,54.2
BEGIN DESCRIPTION:
Structure XS 3
END DESCRIPTION:
XS GIS Cut Line= 6
2229508.75325674657173.7557311352229793.19231157656954.058401477
2229890.83556919657025.1681651832229956.12070031657085.731820261
2230065.44686758657172.078602052 2230268.7796118657100.355065564
#Sta/Elev= 30
       0 2475.07    19.5 2463.49    31.4 2460.71    45.6 2450.78    68.4 2440.99
   173.9 2405.17     230 2390.74   287.4 2371.37   313.7 2365.59   322.2 2359.99
     345 2360.34   353.6 2361.91   359.4 2359.19   382.9 2354.63   514.8 2347.32
   563.9 2346.76   574.6 2345.54   583.1 2342.36   594.8 2340.36  605.332342.351
     697 2344.93   758.1 2353.17   775.1 2352.27   804.8 2354.44   813.3 2358.16
   826.2 2369.13   830.2 2371.07   898.1 2390.53   910.8 2391.61   924.2 2397.01
#Mann= 5, -1 ,  0
       0     0.1       0     290    0.06       0   583.1   0.045       0
  605.33    0.06       0  818.56     0.1       0
#XS Ineff= 2 , 0
                          615.16         2369.21
Permanent Ineff=
       F       F
Bank Sta=583.1,605.33
XS Rating Curve= 0 ,0
Exp/Cntr(USF)=0,0
Exp/Cntr=0.3,0.1

Type RM Length L Ch R = 1 ,30002   ,274.4,264,246.6
BEGIN DESCRIPTION:
Structure XS 2 Disconnected without IFA
END DESCRIPTION:
XS GIS Cut Line= 6
2229524.67335309657223.6386997052229788.94695254657034.720222994
2229982.11078828657171.6330516222230030.93241709657221.516020192
2230077.63136639657249.1108538692230290.96065751657164.203673324
#Sta/Elev= 30
       0 2481.64    12.9 2478.55    30.1 2469.41    38.7 2462.75    52.4 2460.75
    61.6 2450.63    73.1 2443.73   124.7 2428.08   161.6 2412.91   215.7 2394.18
   233.7 2391.73   304.2 2369.95   324.9 2365.39   440.8 2350.73   475.9 2350.13
   495.1 2345.26   505.3 2340.37     524 2339.39   530.1 2340.37   569.8 2341.86
   632.9 2339.86   660.7 2345.78   678.8 2343.04     697 2347.13   735.8 2347.62
   748.7 2355.95   787.4 2366.65   839.1 2385.72   856.3 2388.52   915.3 2408.02
#Mann= 5, -1 ,  0
       0     0.1       0     310    0.06       0   505.3   0.045       0
   530.1    0.06       0  785.66     0.1       0
#XS Ineff= 2 , 0
                          568.84         2349.05
Permanent Ineff=
       F       F
Bank Sta=505.3,530.1
XS Rating Curve= 0 ,0
Exp/Cntr(USF)=0,0
Exp/Cntr=0.3,0.1

Type RM Length L Ch R = 1 ,29738   ,388.2,389,390.6
BEGIN DESCRIPTION:
Structure XS 1
END DESCRIPTION:
XS GIS Cut Line= 3
2229776.52939801657494.0188201542230144.88302863657316.498998168
2230302.43187065657252.148062698
#Sta/Elev= 30
       0 2418.58    35.1  2403.9      44 2401.87    63.3 2391.24      84 2388.37
   146.1  2363.1   177.2 2352.15   189.1 2346.11   201.1 2334.92   204.6 2332.93
   221.6 2332.51   230.5 2334.86   239.4 2336.05     273  2336.6   283.8 2335.64
     294 2336.62   323.7 2336.12     333 2334.23   345.9 2335.86   350.4 2337.09
   362.9 2344.45   368.1  2346.2   403.7 2349.13   426.2 2361.29     447 2366.28
     460 2370.94   472.9 2371.51   515.2 2386.84   537.8 2393.04   579.1  2410.3
#Mann= 5, -1 ,  0
       0     0.1       0   201.1   0.045       0   230.5     0.1       0
   438.9    0.06       0   468.9     0.1       0
#XS Ineff= 2 , 0
                          291.55         2361.21
Permanent Ineff=
       F       F
Bank Sta=201.1,230.5
XS Rating Curve= 0 ,0
Exp/Cntr(USF)=0,0
Exp/Cntr=0.3,0.1

Type RM Length L Ch R = 1 ,29349   ,426.8,409.4,390.7
BEGIN DESCRIPTION:
Structure XS 4
END DESCRIPTION:
XS GIS Cut Line= 3
2229847.53732681 657731.451582062230260.27091292657691.509622113
2230433.35273936657613.844699994
#Sta/Elev= 30
       0 2420.88    36.8    2403    56.9 2395.28    64.9 2390.03      77 2388.93
    93.1  2381.7   113.2 2377.38   158.4 2359.89   177.5 2347.19   185.9 2337.33
   201.6 2332.35   213.6 2324.51     286 2328.77     294 2326.27   318.5 2327.13
   332.92324.494   338.2 2323.26   350.3 2324.35   362.3 2324.28   374.4 2333.39
   378.4 2334.24   402.5 2334.51   440.9 2348.61   475.9 2356.14   493.5 2365.19
   516.2 2367.29   527.8 2373.94   554.9 2381.31   576.7 2391.87   604.4 2399.74
#Mann= 5, -1 ,  0
       0     0.1       0   332.9   0.045       0   350.3     0.1       0
  424.66    0.06       0  534.66     0.1       0
#XS Ineff= 2 , 0
          317.85 2342.43
Permanent Ineff=
       F       F
Bank Sta=332.9,350.3
XS Rating Curve= 0 ,0
Exp/Cntr(USF)=0,0
Exp/Cntr=0.3,0.1

Type RM Length L Ch R = 1 ,28939   ,83.2,84.4,85.5
BEGIN DESCRIPTION:
Structure XS 3
END DESCRIPTION:
XS GIS Cut Line= 6
2229925.85978117658141.6975893432230178.45864329658127.900172504
2230199.68543842658067.4038063662230203.93079745657997.355382417
2230203.93079745657859.381214032 2230492.6152113657775.535373245
#Sta/Elev= 30
       0  2386.9    26.4 2381.15    42.4 2374.85    66.4 2374.22    98.5 2363.39
   158.6 2348.84   186.6 2344.37   222.6 2329.19   246.7 2322.17   260.1 2320.02
     294 2321.49   327.5 2315.15   339.4  2313.1  353.132315.052   375.4 2317.78
   463.4  2318.9   475.4 2321.36   507.4  2321.2   529.7 2323.34   571.3 2322.04
   583.8  2326.2   630.5 2334.33   696.3 2357.09   712.9 2358.44   721.3 2363.76
   750.4 2374.83   783.7 2385.34   795.1 2391.28   812.9 2393.28   825.9 2400.45
#Mann= 7, -1 ,  0
       0     0.1       0     250    0.05       0  302.98     0.1       0
   327.5   0.045       0  353.13     0.1       0  595.24    0.06       0
  785.24     0.1       0
Bank Sta=327.5,353.13
XS Rating Curve= 0 ,0
Exp/Cntr(USF)=0,0
Exp/Cntr=0.3,0.1

Type RM Length L Ch R = 1 ,28855   ,281.1,295.2,305.7
BEGIN DESCRIPTION:
Structure XS 2
END DESCRIPTION:
XS GIS Cut Line= 6
2229941.77987752658206.4393145082230249.56840699 658192.64189767
2230278.22458043658094.998640043  2230288.837978658007.968779985
2230283.53127921657891.221406737 2230507.4739679657815.866284003
#Sta/Elev= 30
       0 2383.79    26.5 2376.24    50.4 2373.68    66.5 2368.07   106.5 2359.52
   138.5 2348.68   174.6 2342.22   214.6 2331.89   222.6  2332.3   250.6 2321.68
   278.7 2321.81   290.7 2316.29   315.9 2314.69   418.9 2312.97     424 2311.61
   431.8 2309.98   445.6 2311.57   478.5 2316.95   504.3 2316.55   569.8 2319.65
   640.4 2326.97   699.5 2342.23   737.5 2357.83   750.1 2358.72   758.6 2364.28
   783.9 2375.01   793.4 2376.13   821.5 2387.43   834.5 2394.91   850.7 2398.64
#Mann= 6, -1 ,  0
       0     0.1       0     230    0.05       0     424   0.045       0
   445.6     0.1       0   634.4    0.06       0   804.4     0.1       0
#XS Ineff= 2 , 0
          418.05 2333.62
Permanent Ineff=
       F       F
Bank Sta=424,445.6
XS Rating Curve= 0 ,0
Exp/Cntr(USF)=0,0
Exp/Cntr=0.3,0.1

Type RM Length L Ch R = 1 ,28560   ,304.3,303.9,302.6
BEGIN DESCRIPTION:
Structure XS 1
END DESCRIPTION:
XS GIS Cut Line= 2
2230111.59806201658414.9028967052230686.31848569658193.003119223
#Sta/Elev= 30
       0 2374.14    26.3 2362.62    39.2 2358.73    73.5 2334.49   116.2 2331.75
   150.7 2326.54     155 2325.35   172.1 2313.64     185 2309.85   205.9 2308.92
   233.8  2309.9   270.4  2308.5   283.6 2309.81   335.9 2309.25   347.9 2308.38
   356.5 2306.53  382.63 2304.77   388.5 2303.36   397.7 2302.99   403.7  2303.1
     408 2304.72   420.8 2311.36   446.5 2331.21   459.4 2339.22   471.2 2344.51
   523.7 2359.06     549 2363.66   562.3 2368.98   579.5 2370.78   616.1 2379.79
#Mann= 6, -1 ,  0
       0     0.1       0      60    0.05       0     170     0.1       0
  382.63   0.045       0     408     0.1       0     590    0.06       0
#XS Ineff= 2 , 0
          371.87 2312.39
Permanent Ineff=
       F       F
Bank Sta=382.63,408
XS Rating Curve= 0 ,0
Exp/Cntr(USF)=0,0
Exp/Cntr=0.3,0.1

Type RM Length L Ch R = 1 ,28256   ,424.1,447.7,467.7
XS GIS Cut Line= 2
2230233.64293963 658725.562585182230810.58236108658445.968865552
#Sta/Elev= 30
       0 2362.29    20.6 2361.03    42.8 2350.45      65 2348.59      74    2339
    78.4 2336.43     101 2331.72   122.8  2324.5   140.6  2316.1   153.9 2314.24
   162.8 2309.78   202.8 2302.88   271.6 2298.17   282.8 2298.82   296.2 2294.29
   309.5  2296.4   318.4 2300.44   331.7 2301.96     354 2299.03   367.3 2299.11
   371.7 2296.86  394.21 2296.88   407.3 2302.69   420.6 2313.45   441.1 2323.02
   509.5 2346.85   522.9 2349.47   556.1 2363.37   571.8 2364.79   641.1 2394.95
#Mann= 4, -1 ,  0
       0     0.1       0   371.7   0.045       0  394.21     0.1       0
     590    0.06       0
#XS Ineff= 2 , 0
          363.55 2319.99
Permanent Ineff=
       F       F
Bank Sta=371.7,394.21
XS Rating Curve= 0 ,0
Exp/Cntr(USF)=0,0
Exp/Cntr=0.3,0.1

Type RM Length L Ch R = 1 ,27808   ,393.9,375.4,357.8
XS GIS Cut Line= 6
2230282.69048949658911.5257541662230674.49357214658852.821851695
2230684.03010561658893.8729125232230702.64340785658955.353213848
2230722.94882847659038.8310541792230966.73636528658941.697211065
#Sta/Elev= 30
       0 2364.51     9.6 2358.35    17.7 2356.53    25.8 2351.79    49.1 2344.04
    58.1 2338.94    82.4 2334.36    94.8 2327.72   151.1 2307.92   163.3 2306.93
   175.4 2302.96   203.9 2298.57     224 2293.03   240.1 2291.02   276.5 2290.97
   296.8 2293.67   361.5 2292.58   381.7 2290.33   441.8 2289.02  460.57  2287.1
  488.732287.102   581.6 2286.39   598.5 2286.84     620 2291.95   641.5 2300.65
   671.7 2304.19   720.1 2314.04   738.6 2320.88   749.2 2322.28     851  2360.4
#Mann= 4, -1 ,  0
       0     0.1       0  460.57   0.045       0  488.73     0.1       0
  838.55    0.06       0
Bank Sta=460.57,488.73
XS Rating Curve= 0 ,0
Exp/Cntr(USF)=0,0
Exp/Cntr=0.3,0.1

Type RM Length L Ch R = 1 ,27433   ,369,368.1,366.8
XS GIS Cut Line= 3
2230337.93583504659373.5099354282230877.15229433659262.560046687
2231050.23412076659138.296171297
#Sta/Elev= 30
       0 2354.55    14.5 2347.49      39 2346.52   107.2 2333.47   116.6 2328.51
   128.9 2329.58   149.3 2323.85   157.5 2317.19   161.6 2315.73   177.9 2318.56
   198.3 2309.71   239.8  2302.3   251.4 2297.82   271.8 2283.76     280  2280.1
   341.2 2283.35   398.4 2281.68   422.9 2284.33  431.082280.753   439.1 2278.85
   449.8 2281.03   484.2 2283.47   506.8 2288.32   540.7 2289.72   559.2 2298.66
   651.1 2311.97   667.5 2317.13   676.9 2317.25   726.6 2335.89   763.6 2352.55
#Mann= 3, -1 ,  0
       0     0.1       0  431.08   0.045       0   449.8     0.1       0
#XS Ineff= 2 , 0
          421.08 2305.34
Permanent Ineff=
       F       F
Bank Sta=431.08,449.8
XS Rating Curve= 0 ,0
Exp/Cntr(USF)=0,0
Exp/Cntr=0.3,0.1

Type RM Length L Ch R = 1 ,27065   ,285.5,294.2,292.8
XS GIS Cut Line= 3
2230491.04668151659752.9585549222230930.40824092659613.161695109
2231059.11011186659597.628710685
#Sta/Elev= 30
       0 2350.47    72.5  2321.3    80.9 2316.12    97.7 2313.38   114.5 2303.86
   134.5 2289.62   139.7 2285.14   148.1 2275.25   152.3 2272.67   185.9 2270.59
   236.2 2270.72   248.8 2273.48   265.6 2274.74   290.8  2272.7   299.2 2273.55
     316 2277.38   328.6 2275.25   374.8 2275.22   387.4 2272.32     400 2271.21
  413.032272.264   425.1 2276.55   499.1  2293.8   523.3 2302.25   531.8 2306.82
   547.5 2309.94   555.5 2313.34   579.7  2313.9   587.7    2319   590.7 2319.93
#Mann= 4, -1 ,  0
       0     0.1       0   387.4   0.045       0  413.03     0.1       0
   590.7    0.06       0
#XS Ineff= 2 , 0
          314.95 2301.38
Permanent Ineff=
       T       F
Bank Sta=387.4,413.03
XS Rating Curve= 0 ,0
Exp/Cntr(USF)=0,0
Exp/Cntr=0.3,0.1

Type RM Length L Ch R = 1 ,26770   ,248.3,249.8,247.4
XS GIS Cut Line= 2
2230506.40737754659974.3916118812231102.31898514659827.822905556
#Sta/Elev= 30
       0 2357.92    51.3 2337.04    71.8 2331.29    84.2 2324.84    92.4 2322.64
   100.7 2317.13     113 2316.02   129.5 2307.78   166.6 2294.46   175.6 2289.21
   191.3  2275.2   197.5 2271.96   228.4 2266.01   244.9  2268.4   281.9 2269.11
   313.2 2265.81   335.5 2267.19     352 2264.36   359.5 2263.04  367.642264.399
     389 2264.93   397.3 2267.65     422 2266.67   450.8 2277.24   490.8 2281.97
   516.7 2287.15   541.4 2295.83   554.6 2296.73   566.2 2301.31   613.7 2313.15
#Mann= 3, -1 ,  0
       0     0.1       0     352   0.045       0  367.64     0.1       0
#XS Ineff= 2 , 0
          251.19 2283.62  401.81          2281.9
Permanent Ineff=
       F       F
Bank Sta=352,367.64
XS Rating Curve= 0 ,0
Exp/Cntr(USF)=0,0
Exp/Cntr=0.3,0.1

Type RM Length L Ch R = 1 ,26521   ,196,197.6,194
XS GIS Cut Line= 2
2230589.32435082660210.7067411752231149.45570698660011.476346272
#Sta/Elev= 30
       0 2354.65    24.3 2345.66    41.2  2337.8    49.7 2335.32    58.2 2329.45
    79.4 2326.64    87.9  2320.6    96.4 2318.58     113 2309.97   138.9 2300.63
   166.3 2286.86   178.8 2284.41   198.3 2274.83   211.1 2266.44   219.5 2263.24
   235.2 2259.77     254 2261.47   282.1  2260.6   304.5 2257.95   334.2 2260.25
   346.9 2257.64   362.6 2256.32  370.622257.618   380.9 2259.39   406.3 2273.81
   419.1 2278.21   448.8 2281.07   512.5 2290.45   525.2 2290.89   594.5 2302.52
#Mann= 3, -1 ,  0
       0     0.1       0   346.9   0.045       0  370.62     0.1       0
#XS Ineff= 2 , 0
           247.8  2284.9
Permanent Ineff=
       F       F
Bank Sta=346.9,370.62
XS Rating Curve= 0 ,0
Exp/Cntr(USF)=0,0
Exp/Cntr=0.3,0.1

Type RM Length L Ch R = 1 ,26323   ,237.8,238.8,239.5
XS GIS Cut Line= 2
2230680.77436815660400.138919936 2231185.3824995660176.412984675
#Sta/Elev= 30
       0 2357.38      30 2344.07    34.3 2341.62    38.7 2337.34    43.1 2334.52
    51.9 2333.69      65 2328.91    74.5 2322.91   101.8 2309.05   152.5 2289.03
   178.7 2275.12   200.6  2265.2   226.9  2258.6   259.5 2257.19     275 2255.07
   283.8 2255.16   301.3 2257.25   320.1 2253.67   336.3 2252.69     345 2253.68
   372.5  2256.4   377.7 2259.27   389.8 2268.84   419.4 2276.31   476.3 2286.76
   493.8 2286.46   506.9 2291.15     520 2292.87   537.5 2298.11     552 2300.48
#Mann= 4, -1 ,  0
       0     0.1       0   320.1   0.045       0     345     0.1       0
     520    0.06       0
Bank Sta=320.1,345
XS Rating Curve= 0 ,0
Exp/Cntr(USF)=0,0
Exp/Cntr=0.3,0.1

Type RM Length L Ch R = 1 ,26084   ,240,237.1,237.5
XS GIS Cut Line= 2
2230764.40623593660587.3599947372231292.86396964660371.243265975
#Sta/Elev= 30
       0 2326.88    32.1 2318.56    79.7 2308.86   125.1 2296.54   146.7 2289.56
   155.3 2283.11     164 2278.93   200.3 2267.34   219.3 2264.28   225.4 2262.27
   240.7 2252.81   246.1 2250.53   262.2 2249.55   268.3 2247.12   276.3 2245.95
   289.8 2247.15   314.4 2250.33   332.5 2254.26   345.5 2254.28   357.3 2252.77
   371.4 2253.14   394.1 2251.07   417.9 2251.35   436.2 2258.07   455.4 2269.79
   470.8 2272.09   501.1 2283.23   535.2 2292.82   548.6 2299.56   570.9 2300.89
#Mann= 4, -1 ,  0
       0     0.1       0   268.3   0.045       0   289.8     0.1       0
     530    0.06       0
Bank Sta=268.3,289.8
XS Rating Curve= 0 ,0
Exp/Cntr(USF)=0,0
Exp/Cntr=0.3,0.1

Type RM Length L Ch R = 1 ,25847   ,441.4,444.3,446.5
XS GIS Cut Line= 4
2230845.89362697660711.2098427842231032.89325384660715.122645238
2231203.05538153660653.3691026292231420.06263636660646.443864139
#Sta/Elev= 30
       0 2303.28    26.3 2296.88    38.3 2289.27    42.3 2288.33    62.3  2289.2
    70.3 2285.82    90.3 2285.87    98.3 2280.22   114.3 2273.18   134.3 2270.86
   158.3 2258.49   166.3 2256.65   182.3 2255.38     199 2247.06   244.2 2247.87
   271.4 2244.93   305.4 2245.38     331 2243.98   339.5  2243.2   344.1 2243.99
   352.2 2246.42   389.2 2247.37   409.2 2245.42   421.2 2247.21   473.2 2289.56
   501.3 2290.96   505.3 2292.72   513.7 2300.66   569.3 2319.09   585.2 2323.11
#Mann= 5, -1 ,  0
       0     0.1       0     331   0.045       0   344.1     0.1       0
  418.06    0.06       0  518.06     0.1       0
#XS Ineff= 2 , 0
                          389.59         2253.09
Permanent Ineff=
       F       F
Bank Sta=331,344.1
XS Rating Curve= 0 ,0
Exp/Cntr(USF)=0,0
Exp/Cntr=0.3,0.1

Type RM Length L Ch R = 1 ,25403   ,221,221,222.7
XS GIS Cut Line= 3
2230799.48737221660977.8453266242231208.33171944661060.027293797
2231376.23605469661054.747292893
#Sta/Elev= 30
       0 2321.44      17 2315.31    30.6 2313.96    61.9 2301.47    86.4 2290.32
   102.7 2277.08   112.1 2273.61     119 2272.65   135.3 2274.82   155.7 2266.03
   176.7 2266.16   192.5 2255.36   216.9 2246.41   245.5 2245.28   261.8  2237.7
   302.6 2237.94   309.6 2235.51   314.9 2234.29   328.12235.513   416.9 2238.16
   436.9 2235.93   467.6 2252.76   484.9 2258.73   496.9 2265.71     509 2267.77
   520.9 2273.32   536.9  2284.7   564.9 2287.27   576.9 2294.91     585 2297.48
#Mann= 4, -1 ,  0
       0     0.1       0   309.6   0.045       0   328.1     0.1       0
  467.02    0.06       0
#XS Ineff= 2 , 0
                           417.1         2248.67
Permanent Ineff=
       F       F
Bank Sta=309.6,328.1
XS Rating Curve= 0 ,0
Exp/Cntr(USF)=0,0
Exp/Cntr=0.3,0.1

Type RM Length L Ch R = 1 ,25182   ,266.3,264.5,263.3
XS GIS Cut Line= 3
2230816.39790735661179.1719849642231152.13324035661272.323252604
 2231337.9252516661272.960459263
#Sta/Elev= 30
       0 2313.08    27.4 2300.75    37.2 2298.54    53.7 2289.23    66.2 2287.36
    78.6 2276.64    89.2 2272.34   107.7 2260.57   124.9 2253.17   136.8 2249.54
   160.7 2247.74   170.4  2241.5   182.4 2236.26   190.82230.555     202 2229.31
   208.32230.469   219.8 2232.38   257.1 2230.33   267.9 2232.62   311.1 2233.89
   323.6 2232.88   360.5 2233.81   384.5 2232.72   396.5 2230.48   420.5 2233.43
   456.9 2251.17   492.5 2263.32   500.5 2267.56   528.5 2271.95   534.2 2274.77
#Mann= 4, -1 ,  0
       0     0.1       0   190.8   0.045       0   208.3     0.1       0
  448.42    0.06       0
#XS Ineff= 2 , 0
                          359.57         2257.93
Permanent Ineff=
       F       F
Bank Sta=190.8,208.3
XS Rating Curve= 0 ,0
Exp/Cntr(USF)=0,0
Exp/Cntr=0.3,0.1

Type RM Length L Ch R = 1 ,24917   ,263.1,264.9,266.1
XS GIS Cut Line= 2
2230788.89786792661481.6724186222231361.54574768661510.790107423
#Sta/Elev= 30
       0  2308.7    15.3 2303.72    35.3  2294.1    71.4 2260.15    75.4 2258.01
    99.4 2254.66   115.4 2249.53   131.4 2246.69   163.5 2248.43   183.5 2241.93
   195.5 2233.53  211.272225.009   219.6 2222.29   231.6 2222.64   235.1 2225.02
   243.6  2229.2   255.6 2228.01   263.6  2229.6     319 2226.92   331.7 2228.53
   395.8 2229.87   419.8 2226.56   431.8 2227.05   435.8 2229.18   443.8 2237.13
   451.9 2242.85   463.9 2245.38   475.9 2252.38     560 2279.99   573.4 2286.29
#Mann= 4, -1 ,  0
       0     0.1       0  211.27   0.045       0   235.1     0.1       0
     560    0.06       0
#XS Ineff= 2 , 0
                          392.57         2241.98
Permanent Ineff=
       F       F
Bank Sta=211.27,235.1
XS Rating Curve= 0 ,0
Exp/Cntr(USF)=0,0
Exp/Cntr=0.3,0.1

Type RM Length L Ch R = 1 ,24652   ,385.1,390,392.8
XS GIS Cut Line= 2
2230736.30237134661711.4253149562231359.84074606661813.499212598
#Sta/Elev= 30
       0 2306.89    48.5 2291.55    60.7  2284.3    68.8 2275.89    72.8 2273.83
   105.3 2267.47   129.6 2251.28   145.8 2248.52   165.1 2240.26   202.5 2237.22
   226.7 2219.51   231.3 2218.89  242.36 2219.52   249.7 2221.72   271.4 2219.52
   279.5 2222.31   304.4 2223.06   324.1 2222.68   344.4 2219.54   417.4 2221.34
   449.8 2219.86   482.2  2222.9   494.4 2227.14     526 2249.45   537.8 2255.65
   567.3 2266.91   579.5 2269.51   607.5 2281.93     620 2283.34   631.8 2283.33
#Mann= 4, -1 ,  0
       0     0.1       0   226.7   0.045       0  242.36     0.1       0
     620    0.06       0
#XS Ineff= 2 , 0
                          316.33          2253.9
Permanent Ineff=
       F       F
Bank Sta=226.7,242.36
XS Rating Curve= 0 ,0
Exp/Cntr(USF)=0,0
Exp/Cntr=0.3,0.1

Type RM Length L Ch R = 1 ,24262   ,253.8,251.2,244.3
XS GIS Cut Line= 2
2230704.27374295661990.3351650612231274.55617108662196.701958119
#Sta/Elev= 30
       0 2256.94     8.4 2253.22    36.5 2244.06    50.9 2241.97    72.2  2243.6
      85  2242.1    89.2 2240.87   102.1 2233.55   178.6 2228.18   246.6 2225.56
   293.4 2225.16   306.2 2223.21   311.4 2220.47   318.9 2213.63   323.2 2211.62
     3442210.804     353 2209.93   361.4 2209.99   366.52211.228   378.5 2221.09
     387 2224.46   408.3 2225.97   433.8 2224.53   523.1 2225.13   548.8 2226.59
   552.9 2227.45   560.9 2231.56     580 2245.46   591.2 2253.59   606.5 2262.26
#Mann= 4, -1 ,  0
       0     0.1       0     344   0.045       0   366.5     0.1       0
     580    0.06       0
Bank Sta=344,366.5
XS Rating Curve= 0 ,0
Exp/Cntr(USF)=0,0
Exp/Cntr=0.3,0.1

Type RM Length L Ch R = 1 ,24011   ,453.2,445.3,436.6
XS GIS Cut Line= 2
2230657.47151462662326.2395534112231247.72492272 662339.55354006
#Sta/Elev= 30
       0 2245.83    38.7  2244.8    66.7  2238.1    94.7 2236.46   126.7 2231.72
   138.7 2225.32   154.7 2226.52   170.7  2217.2   186.8 2210.54   198.8 2208.66
   204.4 2206.61   238.8 2206.37   250.8 2207.98   256.12206.905   262.8 2205.68
   283.72207.131   298.8 2207.66   322.8 2205.92   326.8 2206.52   334.8 2209.76
   358.8 2210.25   370.8 2214.83   380.4 2216.64   420.3 2219.79   430.8 2221.91
   506.8 2231.21   554.8 2239.25   562.8 2241.21   570.8 2244.73   590.4 2246.21
#Mann= 4, -1 ,  0
       0     0.1       0   256.1   0.045       0   283.7     0.1       0
     500    0.06       0
Bank Sta=256.1,283.7
XS Rating Curve= 0 ,0
Exp/Cntr(USF)=0,0
Exp/Cntr=0.3,0.1

Type RM Length L Ch R = 1 ,23566   ,327.2,330.4,337.2
XS GIS Cut Line= 4
2230768.51324056662769.4576733862230945.97200399 662689.42440936
2231026.60444592662637.476337526 2231277.2823955662536.104247315
#Sta/Elev= 30
       0 2243.67    24.1 2243.48    39.1 2240.27    56.7 2238.09    87.4 2226.14
   109.3  2212.3     130 2212.91   144.4  2207.3   163.3  2203.1   175.1  2201.9
   193.5 2202.43   202.1 2201.32   210.82195.761   216.3 2194.63   230.6 2194.47
   240.42195.948   254.2 2197.59   263.9 2196.67   278.2 2197.15   291.4 2200.64
   362.7 2199.22   400.2 2201.23   405.7 2202.61   417.4 2210.36   430.5 2215.43
   476.4 2224.37   490.8 2224.41   512.3 2229.57     532 2236.54     561 2248.97
#Mann= 5, -1 ,  0
       0     0.1       0   210.8   0.045       0   240.4     0.1       0
  430.59    0.06       0  540.59     0.1       0
Bank Sta=210.8,240.4
XS Rating Curve= 0 ,0
Exp/Cntr(USF)=0,0
Exp/Cntr=0.3,0.1

Type RM Length L Ch R = 1 ,23235   ,304.5,299.9,296.6
XS GIS Cut Line= 4
2230965.91220532663072.5792260562231122.89586321662946.965840034
2231211.88516887662919.1849146612231416.36875361662792.985506429
#Sta/Elev= 30
       0 2235.42    23.4 2235.23    64.4 2231.88    84.9 2225.63   107.9 2215.78
   120.7 2209.09   134.9 2209.76   143.5 2205.39   157.7  2200.3   174.8 2195.65
   197.5  2191.1   219.5 2191.57   235.1 2186.98   240.1  2184.5   256.9 2183.83
   264.2 2184.82   269.4 2187.88     282 2188.32   294.6 2195.21   308.7  2200.4
   369.8 2208.43   397.7 2215.48   407.4 2218.96   421.5 2219.75     458  2234.4
   487.8 2244.97   506.1 2252.49   519.8 2259.86   529.6 2262.14   534.6 2264.67
#Mann= 5, -1 ,  0
       0     0.1       0   235.1   0.045       0   269.4     0.1       0
  344.28    0.06       0  514.28     0.1       0
Bank Sta=235.1,269.4
XS Rating Curve= 0 ,0
Exp/Cntr(USF)=0,0
Exp/Cntr=0.3,0.1

Type RM Length L Ch R = 1 ,22936   ,311,313.4,315.1
XS GIS Cut Line= 2
2231059.11011186663338.8589590352231547.28962232663052.608246083
#Sta/Elev= 30
       0 2229.86      27 2227.18    60.5 2226.22    80.1 2224.23      94  2219.6
   107.9 2211.37   117.2 2208.38   126.4 2204.03   135.7 2202.62   145.7 2203.54
   161.5 2197.09   186.7  2194.4   203.7 2190.96  225.962181.427     230 2179.89
   242.4 2179.34   260.9 2181.42   293.4 2183.95   308.9 2187.76   344.4 2191.69
   362.9 2197.53   381.5 2198.47   399.5 2207.04   418.6 2213.08   455.1 2219.03
   469.6  2222.8   478.8 2223.08     502 2228.67   533.2 2239.53   565.9 2252.62
#Mann= 5, -1 ,  0
       0     0.1       0  225.96   0.045       0   260.9     0.1       0
     450    0.06       0  565.91     0.1       0
Bank Sta=225.96,260.9
XS Rating Curve= 0 ,0
Exp/Cntr(USF)=0,0
Exp/Cntr=0.3,0.1

Type RM Length L Ch R = 1 ,22622   ,362.5,372,378
XS GIS Cut Line= 3
 2231143.4320273663562.9777342922231265.47690492663556.320740968
2231658.23951106663389.895907856
#Sta/Elev= 30
       0 2223.31    20.8 2222.84    48.8 2215.79    76.9 2205.34    96.9 2193.27
   112.9  2194.2   116.9 2192.29   122.2 2187.52   128.9 2183.26   140.5 2179.76
     199 2179.61   212.1 2174.85   233.8 2174.95   251.1 2176.14   264.6  2174.3
   272.9 2172.63   290.2 2172.86  294.882174.093   302.3 2181.28   307.6 2184.69
   333.7 2195.06   346.4 2197.84   377.7 2203.18   398.8 2207.83   448.1 2213.95
     464 2214.54   495.9 2220.81   520.5 2223.16   533.5 2225.37   548.8 2226.15
#Mann= 4, -1 ,  0
       0     0.1       0   264.6   0.045       0  294.88     0.1       0
  532.23    0.06       0
Bank Sta=264.6,294.88
XS Rating Curve= 0 ,0
Exp/Cntr(USF)=0,0
Exp/Cntr=0.3,0.1

Type RM Length L Ch R = 1 ,22250   ,369.3,368.7,367.2
XS GIS Cut Line= 2
2231087.95708293663809.2864872972231682.64848658663893.608402741
#Sta/Elev= 30
       0 2219.32    32.5 2219.01    49.6 2215.45    68.9 2209.14   105.3 2191.15
   129.5 2184.54   137.6  2180.7   145.2 2182.63   149.7 2182.38   157.8 2179.88
   169.9 2177.98     178  2175.1   202.2 2172.08   238.6 2170.62  246.152165.536
   262.8 2163.23   270.9 2163.25   282.8  2165.5   311.5 2170.57   323.4 2178.74
   331.5 2182.71   351.7 2197.37   364.5 2201.11   412.3 2207.66   436.5 2209.17
   464.8 2209.36   505.2 2217.48   549.7 2221.24     586 2226.81   600.6 2227.08
#Mann= 5, -1 ,  0
       0     0.1       0  246.15   0.045       0   282.8     0.1       0
     370    0.06       0     470     0.1       0
Bank Sta=246.15,282.8
XS Rating Curve= 0 ,0
Exp/Cntr(USF)=0,0
Exp/Cntr=0.3,0.1
