HEC-RAS study LONGRN.prj: LONGRN

--- LONGRN.g01 (geometry) --- (continued)

Type RM Length L Ch R = 1 ,21881   ,372.1,377,376.6
XS GIS Cut Line= 4
2230965.91220532664153.231142395 2231288.9926563664210.128724705
2231337.59546275664214.3420461162231580.57458894664266.400028911
#Sta/Elev= 30
       0 2214.43    34.8 2215.65    55.1 2214.52   120.1 2198.67   150.4 2187.95
   160.8 2187.67   205.4 2176.95   221.6 2167.01   233.8 2162.46   274.4 2159.61
   294.7 2160.98   323.2 2160.75   332.6 2159.12   338.42156.215   343.3 2154.21
   351.3  2153.9   359.4 2154.08   368.52157.084   383.6 2163.69   391.7 2171.38
   399.9 2177.17   421.8 2184.78   461.3 2192.81   489.9 2205.84   510.4 2211.74
     539 2212.42   555.4 2214.54   575.8 2222.97   604.5 2231.88   625.3 2243.16
#Mann= 5, -1 ,  0
       0     0.1       0   338.4   0.045       0   368.5     0.1       0
  396.84    0.06       0  496.84     0.1       0
Bank Sta=338.4,368.5
XS Rating Curve= 0 ,0
Exp/Cntr(USF)=0,0
Exp/Cntr=0.3,0.1

Type RM Length L Ch R = 1 ,21504   ,333.9,336.6,337.3
XS GIS Cut Line= 2
2230828.33434328664450.5768442212231449.65372023664597.030697359
#Sta/Elev= 30
       0 2210.96    20.4 2209.17    86.1 2209.45   160.1 2188.34   172.4 2182.99
     193 2187.03   242.3 2160.79   275.2 2158.21   283.4 2150.24   287.5 2147.59
   291.4 2147.44   303.9  2147.7   313.5 2150.18   344.6 2152.99   357.4 2152.55
   365.6 2154.83   398.5 2152.74   410.8 2153.43     419 2157.41   443.7 2174.59
   451.9 2177.79     493 2184.97   530.8 2201.09   542.3  2204.7   554.6 2205.41
   567.4 2208.31   587.5 2209.37   600.7 2212.03   616.3 2217.25   638.3 2229.04
#Mann= 7, -1 ,  0
       0     0.1       0   283.4   0.045       0   313.5     0.1       0
     340    0.06       0     540    0.08       0     570     0.1       0
  638.35    0.08       0
Bank Sta=283.4,313.5
XS Rating Curve= 0 ,0
Exp/Cntr(USF)=0,0
Exp/Cntr=0.3,0.1

Type RM Length L Ch R = 1 ,21168   ,466.7,462.2,457
XS GIS Cut Line= 2
2230730.69844119664736.8275571732231345.36082481664940.975352457
#Sta/Elev= 30
       0  2219.6    26.8 2210.78    55.2 2204.08    94.3 2198.47   137.5 2194.49
   200.8  2171.9   229.5 2163.32   254.6 2158.25   267.1 2153.83   279.9 2157.15
   296.6 2152.92   314.7 2144.81  328.482142.916   338.7 2141.96     364  2142.9
   368.2 2143.89   415.9  2142.8   422.3  2145.6   435.7 2155.11   444.4 2159.55
   448.3 2161.02     461 2161.95   477.8 2169.19   503.1  2177.8   526.7 2184.66
     533 2184.67   553.7 2198.39   587.4 2210.65   625.4 2213.15   647.7 2218.53
#Mann= 5, -1 ,  0
       0     0.1       0  328.48   0.045       0     364     0.1       0
     440    0.06       0     550     0.1       0
Bank Sta=328.48,364
XS Rating Curve= 0 ,0
Exp/Cntr(USF)=0,0
Exp/Cntr=0.3,0.1

Type RM Length L Ch R = 1 ,20706   ,502.8,504.5,505.3
XS GIS Cut Line= 3
2230584.24458805665289.358003104 2231161.1840095665300.452991978
2231356.45581369665256.073036482
#Sta/Elev= 30
       0 2216.51    31.2  2212.1   103.9 2194.49     136 2191.41     196 2180.69
     240 2166.34     260 2158.37     288 2151.61     304 2144.22     316 2135.68
     352  2135.8     392 2133.79   396.2 2132.03   404.1 2129.66   419.8 2130.15
     428 2131.98     440 2135.42     456 2136.16     472  2140.7     476 2148.36
     480 2151.56     496 2152.27     512 2157.97     544 2163.19     564 2172.35
   580.1 2182.18   592.4 2187.51   686.8 2201.36   727.8 2211.54   777.3 2228.79
#Mann= 5, -1 ,  0
       0     0.1       0   396.2   0.045       0     428     0.1       0
     470    0.06       0     570     0.1       0
Bank Sta=396.2,428
XS Rating Curve= 0 ,0
Exp/Cntr(USF)=0,0
Exp/Cntr=0.3,0.1

Type RM Length L Ch R = 1 ,20201   ,605.1,608.6,605.8
XS GIS Cut Line= 3
2230504.36066815665755.3475358162231110.14706068 665770.88052024
2231329.82784039665704.310586996
#Sta/Elev= 30
       0 2219.17    35.8 2200.83    63.8 2190.42    91.8 2185.21   155.9 2184.51
   199.9 2179.24   251.9  2164.9   259.9 2160.75   271.9 2160.18   339.9 2140.57
   371.9 2135.06  390.922121.562   403.4 2118.93     416 2121.51   453.8    2124
     480  2121.5     500 2124.77   531.8 2124.66     540 2125.94   552.3 2133.13
     560 2135.07     568 2129.74     576 2129.41     592 2134.57     606 2135.93
     629 2147.62   670.8 2156.74     746 2183.14   771.1 2188.83   835.5 2196.54
#Mann= 6, -1 ,  0
       0    0.03       0      60     0.1       0  390.92   0.045       0
     416     0.1       0     450    0.06       0     550     0.1       0
Bank Sta=390.92,416
XS Rating Curve= 0 ,0
Exp/Cntr(USF)=0,0
Exp/Cntr=0.3,0.1

Type RM Length L Ch R = 1 ,19593   ,445.6,445.6,446.4
XS GIS Cut Line= 4
2230422.25775049666092.6351975892230750.66942116666310.096979522
2231201.12596945666334.5059550452231403.05476696666190.271099682
#Sta/Elev= 30
       0 2199.72    36.4 2195.35      97 2178.18   131.7 2178.64   169.2 2175.35
   195.2  2168.7   229.8 2154.52   275.8 2140.04   307.7 2137.43   333.3 2129.27
   348.7 2128.54   365.4 2123.21   427.4 2118.12   462.8 2110.72   471.5 2108.82
   491.5 2110.77   524.8  2113.9   684.5 2115.38   723.9 2119.31   735.9 2115.05
     804 2126.35   812.4 2131.96     828 2131.73     844 2127.96   859.6 2133.53
   922.5 2138.79    1003 2153.23  1045.4 2165.19  1060.3 2172.97  1093.2    2183
#Mann= 7, -1 ,  0
       0     0.1       0  403.88    0.07       0   462.8   0.045       0
   491.5    0.07       0  603.88     0.1       0  803.88    0.06       0
     905     0.1       0
Bank Sta=462.8,491.5
XS Rating Curve= 0 ,0
Exp/Cntr(USF)=0,0
Exp/Cntr=0.3,0.1

Type RM Length L Ch R = 1 ,19147   ,575.6,583.2,585.9
XS GIS Cut Line= 3
2230466.63770598666729.4875589632231203.34496722666791.619496658
2231407.49276251666900.350387625
#Sta/Elev= 30
       0 2201.45    53.7 2185.14    81.8 2183.96   134.4 2167.13   174.2 2152.09
   182.2 2147.03   190.2 2147.67   230.4 2132.66   266.5 2125.44   286.6  2115.1
  304.462102.378   322.7 2099.95   334.3 2102.31   342.7 2105.14   370.8 2106.12
     423 2104.75   631.8 2105.82   651.8 2113.61   678.6  2119.1     688 2123.08
   736.1 2125.86   749.3 2133.29   794.6 2141.82   810.7 2146.92   823.9 2145.84
   835.4 2153.59   867.2 2157.13   907.9 2167.28   935.1  2179.7   970.6 2185.27
#Mann= 8, -1 ,  0
       0     0.1       0     100    0.07       0     200     0.1       0
  304.46   0.045       0   334.3     0.1       0     690    0.06       0
  859.32     0.1       0  909.32    0.05       0
Bank Sta=304.46,334.3
XS Rating Curve= 0 ,0
Exp/Cntr(USF)=0,0
Exp/Cntr=0.3,0.1

Type RM Length L Ch R = 1 ,18564   ,336.3,337.4,336.8
XS GIS Cut Line= 3
2230479.95169263667219.8860671992230919.31325205667381.872904761
2231048.01512299667408.500878059
#Sta/Elev= 30
       0 2172.95    17.3 2172.95      50 2161.01    59.9 2154.22    72.7 2153.89
    81.2 2148.78   119.5 2131.83   147.6 2125.97   169.4 2115.17   228.6 2095.59
   277.3 2092.78   298.7 2094.86   311.5 2091.31   334.5 2089.22   341.3 2089.45
  346.742091.362   354.1  2095.2   366.9 2095.01   383.9 2100.71   399.9 2102.22
   412.3 2105.78   426.6 2106.19   456.4 2110.51   497.7 2118.58   505.9 2121.99
   518.2 2122.18   530.4 2127.18   554.9 2127.88   566.6 2135.23   599.7 2144.95
#Mann= 4, -1 ,  0
       0     0.1       0   311.5   0.045       0  346.74     0.1       0
  508.27    0.06       0
Bank Sta=311.5,346.74
XS Rating Curve= 0 ,0
Exp/Cntr(USF)=0,0
Exp/Cntr=0.3,0.1

Type RM Length L Ch R = 1 ,18226   ,262.5,258.3,254
XS GIS Cut Line= 3
2230420.03875271667552.7357334222230746.23142561667676.999608812
2230963.69320754667668.123617713
#Sta/Elev= 30
       0 2163.51    15.9 2158.62    25.2 2157.47    68.6 2134.94    77.2 2131.77
    90.3 2129.91   111.4 2118.21   145.7 2107.54   158.5 2102.37   162.8  2100.2
   175.6 2088.39   179.9  2085.7   201.9 2085.76   226.7 2087.54   229.8 2086.68
   235.6 2085.16   245.3  2085.1   262.2 2086.83   282.7 2091.21   299.8 2090.16
   322.8  2091.8   366.1 2100.77   431.1 2104.94   443.1  2107.4   463.1 2114.87
   479.1 2118.78   491.1 2123.17   523.1 2130.85   535.2 2135.65   566.7 2137.59
#Mann= 5, -1 ,  0
       0     0.1       0   229.8   0.045       0   262.2     0.1       0
  459.06    0.06       0  559.06     0.1       0
Bank Sta=229.8,262.2
XS Rating Curve= 0 ,0
Exp/Cntr(USF)=0,0
Exp/Cntr=0.3,0.1

Type RM Length L Ch R = 1 ,17968   ,400.3,394.8,389.7
XS GIS Cut Line= 3
2230377.53354688667867.7961876282230765.85815747 667901.08115425
2230978.88194386667863.358192078
#Sta/Elev= 30
       0  2158.1    30.8 2153.26    58.9 2153.41    62.9 2152.78    70.9 2148.17
    78.9 2146.38      91 2138.37   119.1 2128.09   131.1 2121.52   143.2 2112.37
   147.2  2110.9   159.2 2099.67   181.2 2082.66   187.3 2080.38   195.4 2080.25
   203.4 2080.25   211.62082.837   223.5 2085.22   247.5 2085.29   267.6 2087.14
   319.8 2085.92     360  2096.1     402 2102.04   436.8 2104.33   493.7 2110.93
   505.8 2114.37   526.8 2124.45   554.6 2131.66   566.8 2136.05   606.1 2138.26
#Mann= 4, -1 ,  0
       0     0.1       0   181.2   0.045       0   211.6     0.1       0
  589.75    0.06       0
Bank Sta=181.2,211.6
XS Rating Curve= 0 ,0
Exp/Cntr(USF)=0,0
Exp/Cntr=0.3,0.1

Type RM Length L Ch R = 1 ,17573   ,361,368.9,375.9
XS GIS Cut Line= 3
2230493.26567928668313.8519701862230859.40031213668176.274108147
2231028.04414301668154.084130399
#Sta/Elev= 30
       0 2144.72    20.2 2140.11      33 2138.32    62.9 2127.25    92.8 2118.81
   101.4 2119.73   114.2  2119.4   122.8 2117.58   139.4 2109.32   169.8 2098.77
   191.1  2088.3   203.9 2083.22   217.1 2081.75   280.9  2078.7   293.7 2075.67
   304.1  2073.6   323.6 2073.36   327.9 2073.38   335.1 2075.63   341.3 2078.43
   349.2 2079.67   353.5 2081.33   365.8 2092.96   370.6 2095.09   444.5 2103.52
   496.8 2113.13   508.9 2117.14   537.2 2118.97   545.2 2121.95   561.2  2133.2
#Mann= 4, -1 ,  0
       0     0.1       0   293.7   0.045       0   335.1     0.1       0
  491.13    0.06       0
Bank Sta=293.7,335.1
XS Rating Curve= 0 ,0
Exp/Cntr(USF)=0,0
Exp/Cntr=0.3,0.1

Type RM Length L Ch R = 1 ,17204   ,248.9,251.5,255.1
XS GIS Cut Line= 3
2230482.17069041668566.817716516 2230852.7433188668569.036714291
2231127.89904288668651.139631959
#Sta/Elev= 30
       0 2146.77      50 2126.16     118 2101.74     138 2097.47     166 2098.11
     174 2096.66   179.3  2094.9     206 2080.52     214 2077.06     218 2076.17
     238 2074.45     270 2074.37   285.4 2071.07     298 2068.53     318 2068.73
     326 2071.11     342 2074.31     366 2076.62   374.2 2079.56     395  2089.8
   415.9 2097.96   482.8 2112.28   486.9 2113.46   495.6 2118.81   520.3 2118.75
   528.6 2122.28     537  2124.5   582.9 2132.24   595.3 2135.58   657.7 2147.42
#Mann= 5, -1 ,  0
       0     0.1       0   285.4   0.045       0     326     0.1       0
  480.58    0.06       0  580.58     0.1       0
Bank Sta=285.4,326
XS Rating Curve= 0 ,0
Exp/Cntr(USF)=0,0
Exp/Cntr=0.3,0.1

Type RM Length L Ch R = 1 ,16953   ,351,353.3,356.6
XS GIS Cut Line= 3
2230408.94376384668757.651525151 2230826.1153455 668826.44045617
2231054.67211631668906.324376064
#Sta/Elev= 30
       0 2148.28    11.4 2142.86    51.9 2129.31    84.4 2122.34   124.9 2108.89
   145.2  2103.7   186.8 2089.14   214.1 2087.92   230.3 2080.41   238.4 2078.44
   263.4 2076.11   299.2 2069.57   319.5 2068.27     3262065.048   335.7 2062.63
     360 2065.04   380.3 2063.64   400.6 2067.11   412.7 2076.79   429.2 2082.17
   492.8 2110.93   501.3 2117.15   505.5 2118.63   530.9 2118.46   564.7 2128.42
   598.7 2134.29   636.9 2136.38   641.1  2139.3   649.5 2149.69   664.9 2157.88
#Mann= 5, -1 ,  0
       0     0.1       0     326   0.045       0     360     0.1       0
   462.8    0.06       0   562.8     0.1       0
Bank Sta=326,360
XS Rating Curve= 0 ,0
Exp/Cntr(USF)=0,0
Exp/Cntr=0.3,0.1

Type RM Length L Ch R = 1 ,16600   ,459.9,465.9,472.9
XS GIS Cut Line= 3
2230311.30786175 669019.493262582230812.80135886 669203.67007789
2230999.19717194669188.137093466
#Sta/Elev= 30
       0 2134.41      35 2123.62    73.4 2115.19    86.1 2109.94   104.8 2107.58
   120.2 2101.55   141.5 2095.11   150.1 2088.76   154.3 2087.58   179.9 2087.76
   196.9 2081.85     214 2077.83   252.3 2077.45   282.2 2068.31   333.3  2065.6
   358.9 2062.22   366.6 2058.77   375.9 2056.75   388.5  2057.3   393.82058.707
   400.9 2060.62   414.3 2062.02   486.7 2092.33   499.5    2100   520.8 2101.16
   531.8 2108.45   557.7 2115.78     642 2134.68   682.1 2146.57   721.3 2162.03
#Mann= 5, -1 ,  0
       0     0.1       0   366.6   0.045       0   393.8     0.1       0
     480    0.06       0  684.24     0.1       0
Bank Sta=366.6,393.8
XS Rating Curve= 0 ,0
Exp/Cntr(USF)=0,0
Exp/Cntr=0.3,0.1

Type RM Length L Ch R = 1 ,16134   ,383.9,388.1,391.5
XS GIS Cut Line= 2
2230169.29200416669290.2109911082230621.96755022669767.295512695
#Sta/Elev= 30
       0 2114.04    12.6 2111.12    26.1 2105.03    52.2 2106.11    64.7 2102.28
    75.8 2100.86   119.9  2085.9   143.7 2082.38   185.2 2069.33     196 2068.35
   213.6 2063.24   224.7 2061.79   257.7 2054.76   275.8 2054.14   288.9    2052
   295.6 2049.93   306.4 2049.67   312.2 2049.95     321 2052.03   329.6 2055.49
   334.9 2056.33   358.7 2057.75   397.4 2064.52   422.9 2067.37   428.4 2070.21
   434.2 2074.95     440  2076.8     570 2105.34   620.9 2114.63   657.7 2118.49
#Mann= 5, -1 ,  0
       0     0.1       0   288.9   0.045       0     321     0.1       0
     430    0.06       0     570     0.1       0
Bank Sta=288.9,321
XS Rating Curve= 0 ,0
Exp/Cntr(USF)=0,0
Exp/Cntr=0.3,0.1

Type RM Length L Ch R = 1 ,15746   ,428.3,427.2,426.9
XS GIS Cut Line= 2
2229920.76425338669454.416826445  2230200.357973669978.100301303
#Sta/Elev= 30
       0 2109.44    25.3 2109.02    49.7 2106.93    78.5 2089.96     112  2078.7
   122.8 2072.03   137.6 2072.56   149.4 2068.34   164.2 2065.93     176 2061.21
   185.6 2059.69   202.6    2050   205.6 2049.21   270.5 2049.04   297.9 2047.67
   325.1 2044.42     347 2043.45   352.3 2044.45   356.8 2047.54   368.2 2052.47
     384 2065.88   420.3 2080.23   457.4 2100.53   465.6 2102.08   506.4 2103.37
   510.1 2104.64   520.1 2111.32   542.7 2117.19   574.5 2120.96   593.6 2121.71
#Mann= 4, -1 ,  0
       0     0.1       0   325.1   0.045       0   352.3     0.1       0
     530    0.07       0
Bank Sta=325.1,352.3
XS Rating Curve= 0 ,0
Exp/Cntr(USF)=0,0
Exp/Cntr=0.3,0.1

Type RM Length L Ch R = 1 ,15319   ,378.5,378.7,378.9
XS GIS Cut Line= 2
2229505.81166949669596.4326840332229836.44233793670171.153107712
#Sta/Elev= 30
       0 2105.28    14.7 2102.31    28.5 2105.05    42.4 2105.67    74.7  2102.1
    83.9  2099.3   130.1 2078.91   148.5  2073.8   162.4 2066.86     181 2068.16
   222.4 2056.62     263 2048.18   283.5 2041.47   323.9 2041.48   332.4 2036.29
   341.6 2034.48   362.6 2036.34   402.3  2040.9   435.8 2041.25   438.8 2042.26
   448.5  2052.7   499.2 2071.24   554.6 2086.47   563.9 2090.53   574.3 2091.97
   586.9 2096.99   614.6 2101.86   629.2 2111.95   658.5 2114.12     663 2116.27
#Mann= 4, -1 ,  0
       0     0.1       0   332.4   0.045       0   362.6     0.1       0
     580    0.06       0
Bank Sta=332.4,362.6
XS Rating Curve= 0 ,0
Exp/Cntr(USF)=0,0
Exp/Cntr=0.3,0.1

Type RM Length L Ch R = 1 ,14940   ,421.8,413.5,408.7
XS GIS Cut Line= 3
2229170.74300549669762.8575171452229397.08077852670168.934109938
2229599.00957603 670326.48295195
#Sta/Elev= 30
       0 2104.74    11.2 2102.91    35.8 2094.77    62.2 2088.41    85.1 2087.06
   103.4 2083.51   126.3 2073.54   143.9 2063.77     159 2063.48   176.2 2056.49
   240.9 2047.07   346.1 2042.28   361.5 2032.85     369 2030.69   380.9 2030.87
  387.742032.926   402.7 2038.98     435 2039.19   478.3 2043.17   484.8 2045.32
   499.3 2054.32     510 2055.03   519.6 2059.65   544.2 2064.67   569.3  2072.7
     681 2100.39   709.5 2100.73   712.4 2101.66   717.4 2106.11     721 2107.84
#Mann= 5, -1 ,  0
       0     0.1       0   361.5   0.045       0  387.74     0.1       0
  664.89    0.06       0  694.89     0.1       0
Bank Sta=361.5,387.74
XS Rating Curve= 0 ,0
Exp/Cntr(USF)=0,0
Exp/Cntr=0.3,0.1

Type RM Length L Ch R = 1 ,14526   ,413.1,412.4,412
XS GIS Cut Line= 2
2228804.60837264670155.6201232892229390.42378519670555.039722757
#Sta/Elev= 30
       0 2106.21    23.8 2097.03    41.1 2092.56      67 2088.79    92.9 2080.98
   130.2  2073.6   173.5 2055.92   188.3 2054.33   215.8 2043.61   235.9 2027.56
   245.5 2025.75  264.512027.571   285.1 2031.62   309.3 2029.69   323.8 2026.52
   393.3 2029.08   415.8 2027.49   458.5 2028.11   464.3 2030.19   475.8 2038.25
     503 2048.44   524.7 2049.86   550.6 2057.91   561.1 2058.08   633.7 2075.32
     656 2078.36   677.1 2088.25   701.5 2086.68   706.1 2087.84     709 2090.67
#Mann= 4, -1 ,  0
       0     0.1       0   235.9   0.045       0  264.51     0.1       0
     700    0.06       0
Bank Sta=235.9,264.51
XS Rating Curve= 0 ,0
Exp/Cntr(USF)=0,0
Exp/Cntr=0.3,0.1

Type RM Length L Ch R = 1 ,14114   ,418.5,430.3,434.3
XS GIS Cut Line= 2
2228655.93552173670486.2507917372229206.24696988670839.071437934
#Sta/Elev= 30
       0 2055.98    19.3 2052.97    62.1 2050.08   109.4 2043.87   132.6 2042.89
   166.6 2039.72   185.6 2035.82   223.6 2025.44   228.4 2025.03   237.9 2026.67
     250 2024.15   261.6 2022.95   291.8  2022.8   328.1 2019.58     341 2018.36
   355.5  2019.5   361.4 2022.26   399.4 2021.71   408.9 2022.28   418.4 2024.15
   427.9 2021.06   436.6  2021.7   454.5 2034.16   475.4 2041.87   489.7 2045.52
   509.4 2052.17   523.4 2055.09     618  2081.5   636.4 2088.27   653.7 2089.43
#Mann= 5, -1 ,  0
       0    0.05       0     160     0.1       0   328.1   0.045       0
   355.5     0.1       0     550    0.06       0
Bank Sta=328.1,355.5
XS Rating Curve= 0 ,0
Exp/Cntr(USF)=0,0
Exp/Cntr=0.3,0.1

Type RM Length L Ch R = 1 ,13684   ,458,458.9,454.6
XS GIS Cut Line= 3
2228436.25474202670603.857673803 2228693.6584839671023.248253244
2228884.49229254671112.008164237
#Sta/Elev= 30
       0 2058.69    20.3 2056.18    39.1 2043.95    53.2 2038.66    70.7 2039.36
      94 2037.92   104.8 2039.31   114.3 2034.38   123.6 2032.82   184.6 2033.97
     194 2035.48   226.8 2021.72   233.6 2019.84   277.2 2019.85   290.4  2023.2
   298.1 2023.37   325.4 2022.11   352.8 2016.93   390.6 2016.32   414.6 2013.73
   437.1 2012.54  449.96 2013.76   460.4 2015.73   475.6 2015.74     485 2019.45
   537.6 2031.97   570.7 2038.05   591.9 2043.64   649.3 2052.81   702.5 2066.13
#Mann= 3, -1 ,  0
       0     0.1       0   414.6   0.045       0  449.96     0.1       0
Bank Sta=414.6,449.96
XS Rating Curve= 0 ,0
Exp/Cntr(USF)=0,0
Exp/Cntr=0.3,0.1

Type RM Length L Ch R = 1 ,13225   ,537.5,517.5,495
XS GIS Cut Line= 4
2228060.66618149670941.7136801262228209.47639743671086.935119632
2228273.82904472671177.6237002452228795.73238154671318.374957295
#Sta/Elev= 30
       0 2040.57    55.2 2036.69      70 2030.64    83.1 2022.48    88.7 2020.53
   105.5 2020.46   116.7 2022.19     139  2020.9   177.5 2016.38   199.7 2012.31
   215.6 2011.43   240.2 2012.06     245 2011.05   250.12008.302   254.8 2007.15
     266 2006.73   289.72008.506   297.5 2010.48   321.6 2011.03   487.3 2009.85
   513.2 2015.42   557.7 2019.98   594.8 2022.46   607.4  2024.4   644.7 2026.86
   715.1 2034.02   773.1 2042.01   793.8 2045.85     833 2049.92   859.7 2054.51
#Mann= 4, -1 ,  0
       0    0.07       0      60     0.1       0   250.1   0.045       0
   289.7     0.1       0
Bank Sta=250.1,289.7
XS Rating Curve= 0 ,0
Exp/Cntr(USF)=0,0
Exp/Cntr=0.3,0.1

Type RM Length L Ch R = 1 ,12707   ,348.2,350.7,353.1
BEGIN DESCRIPTION:
Structure XS 4
END DESCRIPTION:
XS GIS Cut Line= 3
2227877.06730277671564.6837103012228176.63200237671617.939656896
2228762.44741492671558.026716976
#Sta/Elev= 30
       0 2164.59    39.7 2149.58    72.2 2131.86    96.6 2116.42   154.9 2088.63
   198.2 2071.11   230.8 2060.56   275.6 2043.48   299.7 2037.01   304.3 2034.97
   311.8 2027.66     336 2025.94   362.9 2007.85   368.1 2004.99     379 2002.26
   392.1 2000.07   408.3 2000.73   412.4 2002.34   444.5 2004.93   468.6 2008.75
   605.4 2008.74   613.4 2007.59   636.5 2018.09   649.6 2025.99   750.1 2044.65
   766.2 2044.47   814.5 2049.23   826.9 2054.47   874.8 2063.89   893.1 2069.61
#Mann= 8, -1 ,  0
       0     0.1       0     230    0.06       0  334.26     0.1       0
     379   0.045       0   412.4     0.1       0  624.26    0.06       0
  804.26     0.1       0  824.26    0.06       0
Bank Sta=379,412.4
XS Rating Curve= 0 ,0
Exp/Cntr(USF)=0,0
Exp/Cntr=0.3,0.1

Type RM Length L Ch R = 1 ,12357   ,103.1,103.8,104.3
BEGIN DESCRIPTION:
Structure XS 3
END DESCRIPTION:
XS GIS Cut Line= 2
2227889.52349233671935.6893554752228768.44632096671980.624060415
#Sta/Elev= 30
       0  2063.8    86.8 2048.03   158.9 2038.37   210.9 2027.59     243 2023.49
     283 2016.28   315.1 2013.95   331.1 2010.56   339.1 2006.41   387.2 2005.45
   391.2 2004.71   399.2 2000.09   407.2 1997.08   415.2 1996.58   427.2  1997.7
   431.2 2000.15   439.2 2002.38   471.3 2002.14   479.3 2004.78   535.3 2003.73
   575.5 2004.66   591.4 2002.66   595.4 2004.03   603.4  2012.9   724.1 2045.24
   756.8 2052.76   773.6 2058.49   787.7 2059.56   859.8 2090.76   880.1 2096.79
#Mann= 6, -1 ,  0
       0     0.1       0     310    0.06       0   399.2   0.045       0
   431.2    0.08       0     510    0.06       0     710     0.1       0
Bank Sta=399.2,431.2
XS Rating Curve= 0 ,0
Exp/Cntr(USF)=0,0
Exp/Cntr=0.3,0.1

Type RM Length L Ch R = 1 ,12253   ,292.6,285,278.8
BEGIN DESCRIPTION:
Structure XS 2
END DESCRIPTION:
XS GIS Cut Line= 2
2227888.28724873672043.1338068912228770.80485376672077.284182645
#Sta/Elev= 30
       0 2078.33     104 2053.09     144  2045.4   194.6  2037.4     212 2033.53
   308.1 2019.05   316.1 2017.05   340.1 2007.67   396.2 2002.26   400.2 2001.34
  407.561996.941   436.2 1996.41   449.91996.975   484.2 2000.03   496.3 1999.44
   516.3 2001.64   540.3 2001.77   560.3 2007.29   580.3 2006.62   604.3 2007.71
     614 2013.75   660.4 2026.16   696.4 2038.18   732.4 2045.63   772.5 2060.82
   784.5 2061.65   796.5 2067.13   828.5 2076.94   840.5 2079.28   883.2 2095.06
#Mann= 6, -1 ,  0
       0     0.1       0     310    0.06       0  407.56   0.045       0
   449.9     0.1       0     610    0.06       0     710     0.1       0
Bank Sta=407.56,449.9
XS Rating Curve= 0 ,0
Exp/Cntr(USF)=0,0
Exp/Cntr=0.3,0.1

Type RM Length L Ch R = 1 ,11968   ,602.2,602.4,603
BEGIN DESCRIPTION:
Structure XS 1
END DESCRIPTION:
XS GIS Cut Line= 4
 2228123.7444521 672478.820528632228382.48002948672336.851496618
2228463.54172283 672309.830932172228718.87156887672204.512033031
#Sta/Elev= 30
       0 2083.81    23.3 2072.16    41.6 2054.01    60.4 2051.28    78.1  2040.4
    96.3 2033.02   128.1 2017.13   141.9 2011.59   160.2 2010.08   173.9 2004.72
   187.6 1996.69   201.2 1995.69   296.9 1998.18     318 1994.31   322.2 1993.51
  369.49 1994.28   381.3 1998.94   390.7 1997.39   406.1 1998.75   420.2 1996.69
   428.9 1998.03   441.8 2003.34   463.5 2016.43   485.1 2017.07   494.9 2021.47
   519.7 2029.16   559.2 2038.56   588.9 2048.79   606.3 2049.41   656.8 2066.91
#Mann= 7, -1 ,  0
       0     0.1       0      60    0.06       0      90     0.1       0
     318   0.045       0  369.49     0.1       0  420.57    0.06       0
  520.57     0.1       0
Bank Sta=318,369.49
XS Rating Curve= 0 ,0
Exp/Cntr(USF)=0,0
Exp/Cntr=0.3,0.1

Type RM Length L Ch R = 1 ,11365   ,502.2,502.6,503.6
XS GIS Cut Line= 2
2228316.11676972673005.2228055962228976.64148458672691.701857988
#Sta/Elev= 30
       0 2079.75     4.5 2076.52    21.1 2071.84    48.1 2059.24   119.6 2031.97
   163.9 2017.48   190.5  1992.6   198.2 1992.94   212.6 1990.45   242.6 1990.48
   389.7 1987.95   405.4 1986.11   416.3 1986.37   425.1 1989.86   438.4 1999.15
   457.2 2009.85   482.7 2010.49   491.5 2013.54   503.8 2014.67     527  2021.9
   549.1  2025.5   584.5  2041.2   603.6 2044.31   630.6 2046.03   648.6 2054.67
   678.7 2063.06   690.4 2069.37   704.1  2071.5   712.9 2078.16   731.2  2081.1
#Mann= 5, -1 ,  0
       0     0.1       0   212.6   0.045       0   242.6     0.1       0
     420    0.06       0     530     0.1       0
Bank Sta=212.6,242.6
XS Rating Curve= 0 ,0
Exp/Cntr(USF)=0,0
Exp/Cntr=0.3,0.1

Type RM Length L Ch R = 1 ,10863   ,686.1,698.1,705
XS GIS Cut Line= 2
2228477.44308256673413.1044267572229141.01169012673090.451801063
#Sta/Elev= 30
       0 2070.51    16.4 2064.25    25.3 2059.95    55.9 2049.24   118.7 2023.79
   176.5  2005.3   203.2 1995.61   220.5 1990.63   229.9 1990.42   265.3 1986.91
   283.3 1982.12   318.8 1983.71   341.1 1981.17   367.1 1982.56  375.161979.997
   381.1 1979.14   398.9 1978.85     409 1979.96   416.7 1982.39   444.9 1984.86
   496.7 2001.16     519 2001.05   527.9 2006.65   532.3 2007.98   563.5 2014.25
   590.1  2020.6   603.6 2022.05   621.8 2027.79   661.3 2036.93   737.9 2061.37
#Mann= 5, -1 ,  0
       0     0.1       0  375.16   0.045       0     409     0.1       0
     460    0.06       0     620     0.1       0
Bank Sta=375.16,409
XS Rating Curve= 0 ,0
Exp/Cntr(USF)=0,0
Exp/Cntr=0.3,0.1

Type RM Length L Ch R = 1 ,10165   ,534.1,535.1,520.6
XS GIS Cut Line= 4
2228512.30904705673710.6281963062228757.18063123673802.079644755
2229199.31075814673894.3612120612229578.75937763673708.631098308
#Sta/Elev= 30
       0 2059.08    42.3 2038.31    93.8 2018.74   154.2 2007.35     192 2002.27
     235 1991.27   264.5 1985.83   284.9 1976.59   309.4 1973.86   329.8 1976.81
   366.6 1978.08   423.8 1977.67     439 1975.92   476.9 1977.89   538.2 1975.11
   588.21976.489   603.6 1974.39   615.91976.528   628.1 1981.99   668.1 1980.84
   687.7 1982.02   720.6 1989.24   740.7 1989.24   864.1 1996.93   918.9 2002.16
   952.3 2003.27   980.7 2007.74  1025.8 2008.63  1061.4 2019.45  1135.5 2031.26
#Mann= 4, -1 ,  0
       0     0.1       0   588.2   0.045       0   615.9    0.06       0
  701.39     0.1       0
Bank Sta=588.2,615.9
XS Rating Curve= 0 ,0
Exp/Cntr(USF)=0,0
Exp/Cntr=0.3,0.1

Type RM Length L Ch R = 1 ,9630    ,556.7,559,552.1
XS GIS Cut Line= 4
2228320.91169151674409.9741852972228638.45027309674198.281797579
2229315.46649419674192.2905035872229676.94123171674304.127991438
#Sta/Elev= 30
       0 2097.77    32.8 2086.24    44.7 2079.92    54.8 2077.78   109.6 2051.52
   121.2 2050.32   215.4 2021.56   316.4  1998.6   369.2  1984.2   402.4 1978.23
   431.4 1976.14   443.4 1971.89   488.11970.671   507.4 1968.91  525.53 1970.67
   551.4 1973.31   587.4 1971.32   783.4 1973.68   811.4 1973.17   823.4 1970.34
   831.4 1972.69   947.3 1977.44   979.4 1982.27  1046.6 1984.87    1060 1986.64
  1075.9 1993.59  1261.4 2018.46  1349.4 2033.38  1402.8 2037.82  1437.1  2046.3
#Mann= 7, -1 ,  0
       0    0.08       0     160     0.1       0   488.1   0.045       0
  525.53     0.1       0  831.63    0.06       0 1031.63    0.05       0
 1178.68     0.1       0
#XS Ineff= 2 , 0
          455.07 1977.66  834.99         1974.73
Permanent Ineff=
       F       F
Bank Sta=488.1,525.53
XS Rating Curve= 0 ,0
Exp/Cntr(USF)=0,0
Exp/Cntr=0.3,0.1

Type RM Length L Ch R = 1 ,9071    ,303.6,306.9,304.2
XS GIS Cut Line= 2
2228697.35877354674591.7749748282229338.42723069 674695.62407069
#Sta/Elev= 30
       0 2010.68    71.7 1987.26   104.2  1979.3   136.6 1973.88   160.9  1973.3
   181.1 1971.38   197.4 1967.81   209.5 1967.93   217.6  1966.2   237.3 1964.68
   274.3 1968.77   290.6 1967.99   300.51966.467   314.9  1964.6   325.11966.372
   343.2 1966.67   351.3 1965.51   355.4 1965.79   375.7 1972.11   387.8 1974.36
   432.4    1980   485.1 1984.36   525.6 1991.51   544.2 1993.59   561.6 1997.19
   586.4 1998.18   594.5 2001.91     600 2002.92   618.8 2004.69   649.4  2009.7
#Mann= 5, -1 ,  0
       0     0.1       0   300.5   0.045       0   325.1     0.1       0
     500    0.06       0     600     0.1       0
Bank Sta=300.5,325.1
XS Rating Curve= 0 ,0
Exp/Cntr(USF)=0,0
Exp/Cntr=0.3,0.1

Type RM Length L Ch R = 1 ,8764    ,285.7,287.4,289.2
XS GIS Cut Line= 3
2228682.06237683674886.9189167392229161.36589619 674938.84346467
2229285.18597202674976.788326619
#Sta/Elev= 30
       0 2013.81    47.5 1994.97    58.1 1991.89    90.6 1984.24   118.8 1980.68
   142.9 1979.05   171.1 1974.77   211.3 1970.77   243.6 1970.37   267.7 1967.74
     328 1968.26   359.7 1963.19   372.3 1962.96   392.4 1962.37  400.93 1962.96
   404.5  1963.6   408.5 1965.89   420.6  1977.5   424.6 1980.28   428.6 1981.96
     465  1991.1   480.9 1997.98   501.8 1998.39     506    2001   510.1 2002.78
   535.2 2010.32   577.1 2020.79   589.6 2024.49     598 2025.63   611.6 2029.36
#Mann= 5, -1 ,  0
       0     0.1       0   372.3   0.045       0  400.93     0.1       0
     410    0.06       0  611.61     0.1       0
Bank Sta=372.3,400.93
XS Rating Curve= 0 ,0
Exp/Cntr(USF)=0,0
Exp/Cntr=0.3,0.1

Type RM Length L Ch R = 1 ,8476    ,739.1,732.3,720.9
BEGIN DESCRIPTION:
Disconnected without IFA
END DESCRIPTION:
XS GIS Cut Line= 2
 2228626.1436329675122.5764804252229209.29624812675252.387850252
#Sta/Elev= 30
       0 2024.29    17.3 2018.11    30.8 2017.25    51.3 2010.88      81 2003.97
    92.2 1999.55   107.8 1998.23   133.2 1992.47   170.1 1983.52     207 1972.58
   239.8 1965.38   268.7 1963.02   292.1 1964.72     329 1964.47   391.4 1966.36
   408.81962.061     416  1960.7   426.2 1960.56   439.6  1962.1   444.7    1963
   449.7 1967.38   473.3 1993.01   477.4 1994.02   493.8 1994.29     502 1999.62
   546.9 2014.62   555.3 2018.26   571.7 2020.78   579.9 2024.74   597.4 2030.16
#Mann= 5, -1 ,  0
       0     0.1       0     370    0.06       0   408.8   0.045       0
   439.6    0.06       0     470     0.1       0
#XS Ineff= 2 , 0
          392.72 1970.62
Permanent Ineff=
       F       F
Bank Sta=408.8,439.6
XS Rating Curve= 0 ,0
Exp/Cntr(USF)=0,0
Exp/Cntr=0.3,0.1

Type RM Length L Ch R = 1 ,7744    ,517.2,524.4,524.7
XS GIS Cut Line= 3
2228636.12912289675643.8190577312229025.56323237675516.004785901
2229165.36009218675518.001883898
#Sta/Elev= 30
       0  2030.7      37 2017.79    46.5 2016.33    63.2 2011.52   109.5 1994.87
   143.2 1984.31   163.8 1973.93   179.6 1963.72   189.5 1959.31   202.1 1955.84
   220.8 1954.87   227.8 1953.53   244.2 1952.16   256.9 1952.38  261.761953.481
   268.4 1956.93   277.9 1957.97   282.1 1960.74   286.3 1962.16   303.2 1962.44
   328.6 1961.01   341.1 1962.68   357.1  1966.8   395.8 1973.65   404.2 1975.72
   412.5 1979.34   432.5 1980.16   444.5 1986.07   488.4 2000.73   549.7 2019.61
#Mann= 5, -1 ,  0
       0     0.1       0   227.8   0.045       0  261.76     0.1       0
     370    0.06       0  469.87     0.1       0
Bank Sta=227.8,261.76
XS Rating Curve= 0 ,0
Exp/Cntr(USF)=0,0
Exp/Cntr=0.3,0.1

Type RM Length L Ch R = 1 ,7220    ,329.1,330,330.5
XS GIS Cut Line= 2
2228688.05367082676095.1632051292229195.31656214675999.302501257
#Sta/Elev= 30
       0 2044.32    18.9 2033.25      53 2018.22    85.6 2006.81     106 1997.66
     167 1979.68   178.4 1978.35   187.4 1975.36   199.6 1974.31   232.2 1968.35
   244.4 1963.27   256.6 1951.47   264.7 1950.11  269.781946.951   272.9 1945.18
   285.1  1945.1   305.4 1945.22   313.6 1946.86   321.7 1948.34   329.9 1954.98
     338 1955.91   358.4 1955.56   378.7 1961.03   429.3 1980.21   443.8 1984.23
   468.3  1997.4   480.5 2000.03   488.6 2004.89     509 2011.85   516.2 2016.49
#Mann= 4, -1 ,  0
       0     0.1       0  269.78   0.045       0   313.6    0.06       0
     510     0.1       0
Bank Sta=269.78,313.6
XS Rating Curve= 0 ,0
Exp/Cntr(USF)=0,0
Exp/Cntr=0.3,0.1

Type RM Length L Ch R = 1 ,6890    ,232.5,232.8,232.3
XS GIS Cut Line= 2
2228771.93178671 676402.716296722229247.24111007 676334.81496481
#Sta/Elev= 30
       0 2008.98    12.4 2008.64    16.4 2007.21    24.5    2002    52.8 1988.67
   101.3 1963.94   109.3    1959   125.5 1952.78   145.7 1950.85   190.2 1951.59
   198.2 1948.89   210.4 1947.37   218.4 1942.31   238.6 1944.35   242.7  1944.2
  248.691941.848   262.9 1940.88     279 1941.86   283.1 1942.61   295.2 1948.39
   299.3 1948.98   327.5 1947.64   347.7 1951.73   355.8 1955.22   366.2 1961.68
   397.6 1985.24   412.4 1989.45   428.6 2000.41   456.8 2010.04   480.1 2015.69
#Mann= 5, -1 ,  0
       0     0.1       0  248.69   0.045       0     279     0.1       0
     320    0.06       0     420     0.1       0
Bank Sta=248.69,279
XS Rating Curve= 0 ,0
Exp/Cntr(USF)=0,0
Exp/Cntr=0.3,0.1

Type RM Length L Ch R = 1 ,6657    ,441,442.8,444.8
XS GIS Cut Line= 2
2228845.82441261676626.3912724222229267.21209005676560.487038509
#Sta/Elev= 30
       0 1993.52    14.5  1985.4    26.7 1983.94    41.6  1977.8    59.1 1972.56
    75.3 1968.76   107.6 1963.05   123.8 1958.83   152.2 1947.93   160.3 1946.86
   164.2 1945.62   168.4 1941.44   172.4 1938.94   188.6 1938.25  202.241938.999
   209.7 1941.24   249.3 1943.47   257.4 1944.76   285.8 1944.93   289.8 1945.66
   297.9 1952.28     306  1957.6   310.1 1959.85   318.2 1962.93   330.3 1970.27
   358.7 1982.09   370.3 1986.25   402.2 2000.24   415.3 2004.86   426.5 2007.98
#Mann= 5, -1 ,  0
       0     0.1       0   172.4   0.045       0  202.24     0.1       0
     250    0.06       0     350     0.1       0
Bank Sta=172.4,202.24
XS Rating Curve= 0 ,0
Exp/Cntr(USF)=0,0
Exp/Cntr=0.3,0.1

Type RM Length L Ch R = 1 ,6214    ,316.3,317.9,317
XS GIS Cut Line= 3
2228797.89406067677033.7992638792229201.30785613  677017.8224799
 2229377.0524799676965.897931969
#Sta/Elev= 30
       0  2012.9    30.3 2013.92    46.3 2006.28    66.3 2000.72   116.8 1983.16
   142.4 1972.38   150.4 1971.33   166.4 1963.98   190.4 1958.19   226.5 1942.19
   238.5 1940.76   270.5 1941.64   282.5 1939.78   290.5 1940.76   334.5 1938.07
   347.7  1935.6   366.6 1934.58   378.6  1935.5   386.6 1943.95   398.6 1945.12
   402.6 1946.83   406.7 1950.62   423.4 1956.11   435.9 1964.05   454.9 1965.36
   469.3 1963.88   503.1 1975.07     536 1982.82   548.5 1987.16     587  1995.5
#Mann= 5, -1 ,  0
       0     0.1       0     290    0.06       0   347.7   0.045       0
   378.6    0.06       0  493.73     0.1       0
Bank Sta=347.7,378.6
XS Rating Curve= 0 ,0
Exp/Cntr(USF)=0,0
Exp/Cntr=0.3,0.1

Type RM Length L Ch R = 1 ,5896    ,384.1,329.7,302.3
XS GIS Cut Line= 3
2228803.88535466677329.3697674852229255.22950206677323.378473493
2229383.04377389677259.471337578
#Sta/Elev= 30
       0 2024.18    52.3 2006.43    80.3 2000.02   124.3 1986.46   128.3 1984.72
   140.3 1975.41   148.3 1971.73   164.3 1968.36   184.3 1969.13   188.3  1967.3
   216.3  1947.8   232.3  1940.5   280.3  1933.9   304.3 1934.87  320.58 1932.14
     336 1931.07   352.8 1932.09   360.3 1935.96   388.3 1937.04   400.3 1938.96
   428.3 1940.87   448.3 1946.82   465.9  1955.1   474.8 1956.54   486.5 1960.93
   527.9 1967.95   543.2 1972.22   564.2    1973   577.7 1972.16   594.3 1976.38
#Mann= 5, -1 ,  0
       0     0.1       0  320.58   0.045       0   352.8     0.1       0
     380    0.06       0  481.38     0.1       0
#XS Ineff= 2 , 0
          301.86 1952.63
Permanent Ineff=
       F       F
Bank Sta=320.58,352.8
XS Rating Curve= 0 ,0
Exp/Cntr(USF)=0,0
Exp/Cntr=0.3,0.1

Type RM Length L Ch R = 1 ,5566    ,502.7,571,601.8
XS GIS Cut Line= 6
2228697.99885925 677695.368749582229031.77437263677821.394622441
2229100.54918887677690.7224715832229133.21722659677603.894266079
2229161.58683829 677458.607466772229402.92144745677340.594296672
#Sta/Elev= 30
       0 2021.74     6.6 2019.06    53.6 2004.85   118.4 1991.31   220.4 1964.28
   263.1 1954.35   280.2 1947.85   293.1 1945.36   309.7 1936.61     323 1930.83
   331.5 1928.28   348.7 1927.24     466 1927.96  496.611925.854   524.6 1925.62
   584.5 1925.85   606.9 1927.87     754 1934.13   762.9 1935.68   780.7    1935
   794.1 1936.82   829.7 1939.35   847.5 1944.98   892.1 1956.11     941  1963.4
   967.8 1966.17     977 1970.28   981.1 1971.13  1007.8 1970.51  1015.3 1971.49
#Mann= 7, -1 ,  0
       0     0.1       0     310    0.06       0  422.48     0.1       0
  474.26    0.06       0  496.61   0.045       0   584.5    0.06       0
  886.69     0.1       0
#XS Ineff= 2 , 0
                          608.23         1939.29
Permanent Ineff=
       F       F
Bank Sta=496.61,584.5
XS Rating Curve= 0 ,0
Exp/Cntr(USF)=0,0
Exp/Cntr=0.3,0.1

Type RM Length L Ch R = 1 ,4995    ,442.3,460.5,466.7
XS GIS Cut Line= 2
2228600.18135893677998.3975965942229293.17436401678268.005826235
#Sta/Elev= 30
       0  2008.7    38.6 1997.02   107.2 1979.88   120.2 1974.82   128.8 1973.51
   167.4 1962.11   206.3  1953.9   244.6 1941.11   287.6 1922.89   301.9 1919.41
   316.6 1922.17   343.4 1922.93   364.8 1921.11   386.3  1924.1     460 1925.95
   506.5 1926.92   545.1 1925.08   552.2 1922.92   595.4 1922.92   605.2 1928.42
     618 1942.65   623.2 1946.69   626.6 1948.14     651 1948.49     661 1950.05
   665.3 1952.26   681.9 1967.37     685 1969.09   702.7 1975.87   743.6 1988.27
#Mann= 6, -1 ,  0
       0     0.1       0     310    0.06       0     460     0.1       0
     520    0.08       0   552.2   0.045       0   595.4    0.08       0
Bank Sta=552.2,595.4
XS Rating Curve= 0 ,0
Exp/Cntr(USF)=0,0
Exp/Cntr=0.3,0.1

Type RM Length L Ch R = 1 ,4535    ,403,384.5,359.8
XS GIS Cut Line= 4
2228488.34387108678283.982610214 2228726.4181061678402.848439823
2228814.50580375678520.5116178742229194.03920141678518.006403104
#Sta/Elev= 30
       0  2001.4    35.6 1989.59   119.1 1968.01   192.1 1941.16   214.4 1936.24
   260.2 1930.46     269 1927.19     284 1917.87     299 1915.38     309 1916.72
     319 1915.11     334 1917.32  339.63 1914.91     354 1913.36   375.8 1914.89
   413.1 1919.76   430.8 1917.56   483.9 1920.27   530.8 1920.05   538.8 1921.69
   554.8 1919.97   564.4 1924.94   590.8  1932.6   610.8 1934.56   618.8 1938.91
   654.8 1940.44   662.8 1943.39   686.8 1957.67   712.1 1967.65   792.6  1989.9
#Mann= 6, -1 ,  0
       0     0.1       0     170    0.06       0   336.1     0.1       0
  339.63   0.045       0   375.8     0.1       0  783.08    0.08       0
#XS Ineff= 2 , 0
                          415.37         1934.46
Permanent Ineff=
       F       F
Bank Sta=339.63,375.8
XS Rating Curve= 0 ,0
Exp/Cntr(USF)=0,0
Exp/Cntr=0.3,0.1

Type RM Length L Ch R = 1 ,4150    ,331.3,331.9,332.1
XS GIS Cut Line= 3
2228408.45995119678833.1845594822229107.44425026678735.326757613
2229235.25852209678623.489269761
#Sta/Elev= 30
       0  2008.9    48.2 1992.85    80.5 1979.42    92.6 1976.68   141.5 1956.69
   193.6 1944.71   217.8 1932.65   242.1 1914.29   254.8 1911.78   262.2 1910.18
  303.151911.759   329.3 1914.27   398.9 1915.78   427.8 1920.47   452.1 1917.42
   476.3 1918.42   492.5 1916.46   528.8 1918.34   538.3 1917.28     646 1922.47
   651.7 1924.18   666.1 1932.13   694.4 1932.19   707.8  1938.2   738.7 1946.49
   758.9 1953.54     773  1961.3   791.8 1964.67   807.8 1971.92   875.6 1985.24
#Mann= 6, -1 ,  0
       0     0.1       0   254.8   0.045       0  303.15     0.1       0
     390    0.06       0     490     0.1       0     690    0.08       0
Bank Sta=254.8,303.15
XS Rating Curve= 0 ,0
Exp/Cntr(USF)=0,0
Exp/Cntr=0.3,0.1

Type RM Length L Ch R = 1 ,3819    ,573.1,585.2,591.8
XS GIS Cut Line= 3
2228466.59031026679150.8116800162229274.80634177679064.627582019
2229423.88778022679161.839421806
#Sta/Elev= 30
       0 2035.68     5.6 2035.14    21.7 2028.46      70 2003.61   110.2 1988.21
   138.4 1975.67   162.5 1962.58   178.6 1948.84   202.9 1944.92     247 1908.99
   254.41907.065   270.1 1905.43   289.11906.627   303.3  1907.8   311.3 1910.85
   319.2 1911.22     436 1910.75   448.1 1909.37   460.2  1911.2   512.5 1908.36
   520.5 1909.16     530 1907.38   701.5 1916.62   794.1 1927.11     824 1926.77
   838.3 1933.44   871.7  1935.2   892.2 1942.28   955.8 1954.61   990.8 1963.85
#Mann= 5, -1 ,  0
       0     0.1       0     230    0.06       0   254.4   0.045       0
   289.1    0.06       0     330     0.1       0
#XS Ineff= 2 , 0
                          346.62         1933.26
Permanent Ineff=
       F       F
Bank Sta=254.4,289.1
XS Rating Curve= 0 ,0
Exp/Cntr=0.3,0.1

Type RM Length L Ch R = 1 ,3233    ,309,320.9,329.1
XS GIS Cut Line= 3
2228427.15586195 679375.586668092229049.26299786679546.748799734
2229231.18211802679590.532125236
#Sta/Elev= 30
       0 2029.39    50.8 2022.71    79.9 2015.46   112.7 2000.12   158.7 1982.48
     196 1974.88   212.6  1968.6   233.4 1957.39   254.1  1939.4   278.7 1934.11
   337.1 1904.43   349.5 1905.71   357.8 1903.36   374.4 1903.32   412.1 1906.53
   523.8  1907.3   540.4 1903.15   552.8 1901.77   577.7  1903.1   600.8 1905.86
   610.9 1911.43   623.5 1914.81   639.9 1914.73   652.3 1917.74   672.9 1917.47
     714 1925.24   788.1 1949.66   804.6 1960.02     821 1960.16   832.3 1966.46
#Mann= 5, -1 ,  0
       0     0.1       0     280    0.06       0     480     0.1       0
   540.4   0.045       0   577.7     0.1       0
Bank Sta=540.4,577.7
XS Rating Curve= 0 ,0
Exp/Cntr=0.3,0.1

Type RM Length L Ch R = 1 ,2912    ,380.8,350.8,337.2
XS GIS Cut Line= 3
 2228552.6346737679537.7503286792228847.74255479679814.216363439
2229145.79354972679838.548348801
#Sta/Elev= 30
       0 1962.86    30.4 1949.49    48.7 1932.09    59.7 1924.56    65.1 1922.35
    75.2  1921.6    84.2  1923.3    98.3 1923.24   127.9 1915.95   154.9  1914.1
   174.8 1903.72   191.2 1903.51   202.2 1900.84     254 1901.59   267.9 1903.25
   326.8 1903.18     336 1901.24   344.4 1899.91   373.6 1899.84  381.14 1901.26
   399.5  1904.5   412.8 1902.83   428.9 1902.78   513.2 1912.56   537.4  1916.9
   565.3 1919.11     593 1925.42   649.6 1941.91   661.7 1942.86   703.4 1956.74
#Mann= 5, -1 ,  0
       0     0.1       0      60    0.06       0     190     0.1       0
     336   0.045       0  381.14     0.1       0
Bank Sta=336,381.14
XS Rating Curve= 0 ,0
Exp/Cntr(USF)=0,0
Exp/Cntr=0.3,0.1

Type RM Length L Ch R = 1 ,2562    ,333.2,323.6,321.4
XS GIS Cut Line= 5
2228332.06495023680295.7858962582228542.73565962680109.150083142
 2228748.0053993680025.4169456192228943.33311332679912.451993795
2229178.68496333679910.718359659
#Sta/Elev= 30
       0 2001.45    88.4 1966.41   227.1 1932.18   245.6 1921.43   254.1 1920.82
   265.4  1924.6     278  1920.1   313.2 1919.03     350 1908.82   369.4 1907.59
  384.77 1897.22   399.1 1895.82   422.8 1897.23   429.9 1900.41   477.4 1899.97
   494.7 1901.73   535.6 1900.41   618.9 1900.66   637.3 1902.05   655.7 1900.63
   696.7 1901.26   714.2 1905.64   781.6 1914.36   821.6 1926.81   861.6 1943.24
   889.6 1949.87   901.6 1950.62   909.6 1955.01   933.6 1963.99   964.1  1972.7
#Mann= 5, -1 ,  0
       0     0.1       0  341.45    0.06       0  384.77   0.045       0
   422.8    0.06       0  441.45     0.1       0
#XS Ineff= 2 , 0
                          434.12         1910.03
Permanent Ineff=
       F       F
Bank Sta=384.77,422.8
XS Rating Curve= 0 ,0
Exp/Cntr(USF)=0,0
Exp/Cntr=0.3,0.1

Type RM Length L Ch R = 1 ,2238    ,420.3,433.3,443.9
XS GIS Cut Line= 3
2228565.23214398680567.2248086132229055.60455942680143.484833582
2229234.02032133680083.567615617
#Sta/Elev= 30
       0 2002.15    14.9  1996.1    34.7 1994.48    51.7 1982.93   136.8 1951.05
   193.5 1933.02   235.6 1922.83   253.1 1923.11   266.2  1918.7   315.8 1911.97
   326.8  1908.7     358 1908.01   386.4 1897.24   409.1 1894.15   423.3 1892.88
   449.7 1894.14   458.5 1898.29   471.5 1898.61   606.6 1895.76   638.3 1916.41
   648.1 1919.95   657.1 1920.63   678.2 1930.16   699.3 1936.66     712 1943.35
   724.6 1946.25   737.3 1951.94   779.5 1954.72   792.2 1963.22   836.3 1975.42
#Mann= 5, -1 ,  0
       0     0.1       0     220    0.06       0     370     0.1       0
   409.1   0.045       0   449.7     0.1       0
#XS Ineff= 2 , 0
                          472.07         1904.39
Permanent Ineff=
       F       F
Bank Sta=409.1,449.7
XS Rating Curve= 0 ,0
Exp/Cntr(USF)=0,0
Exp/Cntr=0.3,0.1

Type RM Length L Ch R = 1 ,1805    ,592.7,585.4,574.4
XS GIS Cut Line= 4
2228663.64913329680646.8091638062228889.21107905680559.228056751
2229314.65286542680523.6397704382229452.48287126680458.862271277
#Sta/Elev= 30
       0 2002.84    26.3 1986.57   133.6  1945.5   167.9 1931.26   176.5 1926.12
   185.1 1924.67   193.7 1925.77   219.4 1915.56     261 1905.47   317.2 1900.85
   329.2 1904.77   337.3 1904.96   365.1 1896.91   385.4 1895.12   453.7 1893.09
   477.8 1896.09   501.8 1893.93   517.9 1896.17   566.1 1894.44  577.571889.974
   597.8 1889.19616.06021890.012   630.3 1898.78   654.7 1922.03   670.6  1932.1
     717 1949.01     741  1960.5   754.6 1961.51   768.7 1968.78   821.2 1983.95
#Mann= 5, -1 ,  0
       0     0.1       0     240    0.06       0  341.97     0.1       0
  577.57   0.045       0616.0602     0.1       0
#XS Ineff= 2 , 0
          524.08 1917.17
Permanent Ineff=
       F       F
Bank Sta=577.57,616.0602
XS Rating Curve= 0 ,0
Exp/Cntr(USF)=0,0
Exp/Cntr=0.3,0.1

Type RM Length L Ch R = 1 ,1219    ,483.4,493.8,512.1
XS GIS Cut Line= 2
2228953.66770446681233.6963522852229624.69263157680868.227418772
#Sta/Elev= 30
       0 1978.77    43.5 1964.51    61.2 1961.75    80.3 1955.19    98.5 1947.46
   107.6 1939.56   139.5 1939.77   149.7  1934.6   180.5 1928.38   198.7 1916.98
   220.4 1916.08   248.8 1907.12   332.5 1896.29   352.3 1886.43   370.8 1883.99
   391.5 1884.49   397.4 1886.57   408.2 1892.04   417.3 1892.78   499.3 1887.76
     536  1888.4   562.5 1900.95   571.3 1907.69   585.9 1910.28   595.1 1917.62
   631.4 1934.01   695.2 1956.91     718 1968.08   733.5 1969.63   764.1 1983.78
#Mann= 5, -1 ,  0
       0     0.1       0     150    0.06       0     270     0.1       0
   352.3   0.045       0   397.4     0.1       0
#XS Ineff= 2 , 0
                          449.39         1917.03
Permanent Ineff=
       F       F
Bank Sta=352.3,397.4
XS Rating Curve= 0 ,0
Exp/Cntr(USF)=0,0
Exp/Cntr=0.3,0.1

Type RM Length L Ch R = 1 ,726     ,361.6,369.1,374.4
XS GIS Cut Line= 3
2228957.66190046681349.5280361312229582.75357363   681447.385838
2229776.47207937681381.481604088
#Sta/Elev= 30
       0 1984.53    95.7 1956.36     124 1944.02   156.4    1943   180.7 1930.83
     205 1930.37   221.2 1923.05   233.3 1924.31   261.7 1910.94   277.9 1909.42
   314.3 1894.41     359 1894.68   379.1    1891   427.7 1887.28   516.7 1889.49
   545.1  1886.1   557.2 1889.87   581.5 1882.19   601.8 1880.26     626 1882.29
   642.7 1894.99   654.5 1907.17   663.9 1920.48   676.5 1929.79   727.2 1953.69
   744.1  1964.1   756.7 1965.69   765.2 1971.21   793.2 1978.64   837.3 1994.89
#Mann= 5, -1 ,  0
       0     0.1       0     230    0.06       0     330     0.1       0
   581.5   0.045       0     626     0.1       0
Bank Sta=581.5,626
XS Rating Curve= 0 ,0
Exp/Cntr(USF)=0,0
Exp/Cntr=0.3,0.1

Type RM Length L Ch R = 1 ,356     ,230.1,222.7,214.6
XS GIS Cut Line= 6
2228899.74605854681597.1681878012229351.09020594 681665.06951971
 2229452.9422038681728.9766556252229508.86094772681802.869281527
2229700.58235547681848.8025354662229924.25733117681675.055009697
#Sta/Elev= 30
       0 1994.37    56.6 1976.81    69.2 1975.12    77.3 1970.42    89.4 1969.47
   178.4 1941.73   186.5 1939.13   198.6 1931.36   222.9 1931.35   264.1 1911.97
   275.5 1908.77   279.5 1904.63   299.8  1903.2   311.9 1893.66   315.9 1892.51
   372.6 1889.95   411.8 1890.98   491.6 1881.41   665.7    1876   696.4 1875.78
   702.11876.008   812.5 1885.87     879 1895.93     903 1906.68   954.9 1923.54
  1025.2 1956.85  1056.2 1962.89  1065.5  1968.9  1076.5 1972.87  1152.6 1994.48
#Mann= 5, -1 ,  0
       0     0.1       0     290    0.06       0     390     0.1       0
   665.7   0.045       0   702.1     0.1       0
#XS Ineff= 2 , 0
           614.3 1901.76     720         1906.34
Permanent Ineff=
       F       F
Bank Sta=665.7,702.1
XS Rating Curve= 0 ,0
Exp/Cntr(USF)=0,0
Exp/Cntr=0.3,0.1

Type RM Length L Ch R = 1 ,134     ,,,
XS GIS Cut Line= 3
2228875.78088257 681950.654533332229668.62878751682046.515237202
2229952.21670313681820.843163503
#Sta/Elev= 30
       0 1960.06    24.6 1952.05    44.7 1942.42    60.8 1941.26   145.4 1913.05
   234.1 1897.11   246.2 1893.23   293.8 1890.69   330.8  1883.7   372.9 1881.33
   451.7 1886.09   544.3 1887.19   572.5  1879.1     633 1880.05   645.1 1875.76
   656.8 1874.15  670.621875.734   689.2 1881.11   781.3 1882.05     879 1892.78
   946.3 1895.21   975.7 1906.35  1001.4 1911.14  1038.3 1922.51  1070.6  1926.6
  1089.8 1932.21  1104.8 1941.11  1118.1 1942.97  1140.5  1953.6    1161 1957.16
#Mann= 5, -1 ,  0
       0     0.1       0     210    0.06       0     310     0.1       0
   645.1   0.045       0  670.62     0.1       0
Bank Sta=645.1,670.62
XS Rating Curve= 0 ,0
Exp/Cntr(USF)=0,0
Exp/Cntr=0.3,0.1
LCMann Table=0

Chan Stop Cuts=-1
Use User Specified Reach Order=0
Composite Channel Slope=5
